HEC-RAS study 5238_ras.prj: 5238

--- 5238_ras.g01 (geometry) --- (continued)

Type RM Length L Ch R = 3 ,48828.85,,,
BEGIN DESCRIPTION:
END DESCRIPTION:
Bridge Culvert--1,0,-1,-1, 0
Deck Dist Width WeirC Skew NumUp NumDn MinLoCord MaxHiCord MaxSubmerge Is_Ogee
22.481700,25.000000,2.6,0, 47, 47, , , 0.95, 0, 0,0,,
 9633.50 9645.27 9655.73 9666.18 9676.64 9687.10 9697.55 9708.01 9718.47 9731.88
 9739.38 9749.83 9760.29 9766.10 9770.75 9781.20 9791.66 9800.32 9802.12 9812.57
 9823.03 9833.49 9843.94 9854.40 9868.76 9875.31 9885.77 9896.22 9906.68 9927.59
 9954.64 9954.6410014.6410014.6410066.0710076.4610086.9110097.4910108.0810118.67
10129.2510139.8410145.8710150.4310161.0110171.6010175.39
 1014.35 1011.80 1008.58 1005.49 1003.59 1000.76  998.41  994.08  990.54  983.89
  981.22  979.95  980.11  979.65  978.66  974.92  972.55  971.37  971.05  966.81
  964.76  963.88  963.15  962.17  961.38  960.48  949.82  948.97  948.57  947.60
  946.67  946.67  944.50  944.50  942.66  942.22  941.59  942.16  946.06  948.60
  953.48  959.50  961.54  963.27  972.70  979.88  982.84
   14.35   11.80    8.58    5.49    3.59    0.76   -1.59   -5.92   -9.46  -16.11
  -18.78  -20.05  -19.89  -20.35  -21.34  -25.08  -27.45  -28.63  -28.95  -33.19
  -35.24  -36.12  -36.85  -37.83  -38.62  -39.52  -50.18  -51.03  -51.43  -52.40
  -53.33  943.17  941.00  -55.50  -57.34  -57.78  -58.41  -57.84  -53.94  -51.40
  -46.52  -40.50  -38.46  -36.73  -27.30  -20.12  -17.16
 9633.50 9645.27 9655.73 9666.18 9676.64 9687.10 9697.55 9708.01 9718.47 9731.88
 9739.38 9749.83 9760.29 9766.10 9770.75 9781.20 9791.66 9800.32 9802.12 9812.57
 9823.03 9833.49 9843.94 9854.40 9868.76 9875.31 9885.77 9896.22 9906.68 9927.59
 9979.59 9979.5910039.5910039.5910066.0710076.4610086.9110097.4910108.0810118.67
10129.2510139.8410145.8710150.4310161.0110171.6010175.39
 1014.35 1011.80 1008.58 1005.49 1003.59 1000.76  998.41  994.08  990.54  983.89
  981.22  979.95  980.11  979.65  978.66  974.92  972.55  971.37  971.05  966.81
  964.76  963.88  963.15  962.17  961.38  960.48  949.82  948.97  948.57  947.60
  945.77  945.77  943.60  943.60  942.66  942.22  941.59  942.16  946.06  948.60
  953.48  959.50  961.54  963.27  972.70  979.88  982.84
   14.35   11.80    8.58    5.49    3.59    0.76   -1.59   -5.92   -9.46  -16.11
  -18.78  -20.05  -19.89  -20.35  -21.34  -25.08  -27.45  -28.63  -28.95  -33.19
  -35.24  -36.12  -36.85  -37.83  -38.62  -39.52  -50.18  -51.03  -51.43  -52.40
  -54.23  942.27  940.10  -56.40  -57.34  -57.78  -58.41  -57.84  -53.94  -51.40
  -46.52  -40.50  -38.46  -36.73  -27.30  -20.12  -17.16
BR Coef=-1 , 0 , 0 ,, 0 ,,,0.8,0,1,0,
WSPro=,,,, 1 ,,,, 0 ,,,, 0 ,,,,-1 ,-1 ,-1 , 0 , 0 , 0 , 0 , 0
BC Design=,, 0 ,, 0 ,,,,,,

Type RM Length L Ch R = 1 ,48800.03,247.787900,247.787900,247.787900
XS GIS Cut Line= 2
513633.228242278799206.785486475513853.280325621 799863.03548646
#Sta/Elev= 30
9637.8241018.8159678.1291006.1619762.507984.57759783.602973.81079794.149971.0066
9804.696971.57769836.338965.27039878.527962.78449889.074954.70219899.621949.5711
9931.263948.51499962.904944.07699973.452 933.8579983.999931.074110005.09930.5622
10047.28 933.89710057.83942.575310100.02942.362710121.11947.018110131.66 951.613
10142.21960.581210152.75963.560810173.85978.424110205.491005.47110216.041008.363
10237.131023.61410247.681028.77810268.771033.00110321.511032.18310329.981035.053
#Mann= 3 , 0 , 0
9637.824  0.0438       09637.824  0.0438       010329.98  0.0438       0
#XS Ineff= 2 , 0
       09878.143                       0
Bank Sta=9637.824,10329.98
Exp/Cntr=0.3,0.1

Type RM Length L Ch R = 1 ,48552.25,247.787800,247.787800,247.787800
XS GIS Cut Line= 6
513405.790510279799288.251171947513515.756346447799623.504905004
513554.173603309799722.725607332 513598.13205773799821.306217407
513621.323544581799867.901917541513654.530288675799927.881287463
#Sta/Elev= 30
9681.6641043.9289688.7661035.8029743.3241008.2879772.956989.17999804.528978.5804
9825.575978.23299836.099974.72599846.622966.44769878.194964.32719888.717960.9365
9899.241955.28869909.765954.87439941.336939.6828 9951.86936.92169962.384931.2291
9972.907929.6213    9999930.420910046.82936.924310068.27937.226610078.99940.1352
10089.71947.711510121.88966.291610132.61970.215910143.38978.645610154.33984.0972
10192.03986.825710252.95997.075610297.631002.55710320.37 999.96210369.44999.1204
#Mann= 3 , 0 , 0
9681.664    0.12       09681.664    0.12       010369.44    0.12       0
#XS Ineff= 2 , 0
       0                               0
Bank Sta=9681.664,10369.44
Exp/Cntr=0.3,0.1

Type RM Length L Ch R = 1 ,48304.46,291.470500,291.470500,291.470500
XS GIS Cut Line= 6
513125.685961306799424.968868452513309.036689685799742.276427299
513377.335365922799841.632433017513419.998626068799890.311029454
513468.678427423799937.210876068513582.390948435800032.082556726
#Sta/Elev= 30
9653.3371074.8919699.6861025.5079711.2641011.3689731.341994.4378 9734.42992.1615
9745.998989.60489769.154987.65059792.311968.43369815.467953.79369850.387942.5062
9908.091935.9682 9919.67933.67049931.248935.60089949.592934.68399969.433929.3621
10019.84 930.20710030.93931.271810058.66929.899910070.52930.542910082.51934.2547
10107.37949.4269 10119.8955.581210167.28974.284510197.62975.938310333.86976.8944
10346.78 979.66510372.61982.002210385.53 986.62710398.45983.253710420.91989.4071
#Mann= 3 , 0 , 0
9653.337    0.12       09653.337    0.12       010420.91    0.12       0
#XS Ineff= 2 , 0
       0                               0
Bank Sta=9653.337,10420.91
Exp/Cntr=0.3,0.1

Type RM Length L Ch R = 1 ,48012.99,451.893000,451.893000,451.893000
XS GIS Cut Line= 6
   512861.867523799678.551966459513027.824335689799840.406295654
513092.613591869799917.445777834513132.780876553799948.758997447
513183.947236334799976.660999788513436.344628791800077.119369362
#Sta/Elev= 30
9722.256 1063.469726.6321059.5169731.4911057.4959745.8141055.6059754.5691051.503
9768.5371034.8179796.4741025.3599810.4421015.5369846.0711018.2799852.3481015.647
9894.253981.23659932.006952.54249954.072 938.1729986.931923.561310013.05922.5638
10051.49 929.46310099.74 932.35710108.43931.484610131.69924.236510154.21 924.814
10165.31926.927610176.05933.515410197.52949.884310208.26953.847110283.44956.4752
10358.62956.748610369.36964.171510390.83973.660510412.39976.657710435.87977.4222
#Mann= 3 , 0 , 0
9722.256   0.073       09722.256   0.073       010435.87   0.073       0
#XS Ineff= 2 , 0
       0                               0
Bank Sta=9722.256,10435.87
Exp/Cntr=0.3,0.1

Type RM Length L Ch R = 1 , 47561.1,247.787900,247.787900,247.787900
XS GIS Cut Line= 6
 512805.27959104800312.069866463512952.692562324800308.423689464
513265.182666961800265.863348051  513385.6399633800259.881755864
 513500.12959867800269.854214636513612.564183632800298.448184084
#Sta/Elev= 30
9665.0811039.2989684.8471029.0269714.8821016.7959744.8861012.1279805.072 993.739
9855.537960.9799 9865.64 951.7989875.743939.63469885.847930.98479906.054924.2524
9916.157918.59869946.468920.93989966.674918.61169986.881 919.62810007.08916.6432
10027.26917.725910047.44926.269310077.67931.2574 10097.8939.7159   10128943.5184
10148.06948.8496 10158.1 955.15210178.16956.426510318.38954.716210338.53 966.649
10368.81965.223710378.99970.491410399.37973.633910409.67977.306810479.98 984.823
#Mann= 3 , 0 , 0
9665.081  0.0617       09665.081  0.0617       010479.98  0.0617       0
#XS Ineff= 2 , 0
       0                               0
Bank Sta=9665.081,10479.98
Exp/Cntr=0.3,0.1

Type RM Length L Ch R = 1 ,47313.31,247.787800,247.787800,247.787800
XS GIS Cut Line= 6
512812.303715425800509.904198608512985.631782131800537.312188582
513296.668079114800520.099813077513408.834511468800525.587056533
513516.007067895800543.000520293513624.797738672800574.208765834
#Sta/Elev= 30
9636.867 994.6319691.151995.34329721.651 999.5549752.002998.66899792.108993.0742
9812.161980.97729822.163978.10339842.163965.73579872.179942.47889882.191932.2933
9892.204926.14499942.348916.97639972.468917.71969992.548915.109310022.64 916.618
10042.69922.847210092.79928.386410162.81953.387710243.03954.339510253.12958.0958
 10263.2965.100910273.29 968.37210293.53970.017610334.23996.762610344.411001.489
10354.731003.03510385.751002.39110406.43994.691410427.28981.084910458.66 976.308
#Mann= 3 , 0 , 0
9636.867  0.0811       09636.867  0.0811       010458.66  0.0811       0
#XS Ineff= 2 , 0
       0                               0
Bank Sta=9636.867,10458.66
Exp/Cntr=0.3,0.1

Type RM Length L Ch R = 1 ,47065.52,247.787900,247.787900,247.787900
XS GIS Cut Line= 6
512775.676112912800592.316304257512868.421874444800646.866097947
 513094.74734062800742.835693486513335.193568358800861.167624783
513439.489923818800916.689681955513532.815002075800974.333669898
#Sta/Elev= 30
9591.507 968.9689718.088968.25649750.723965.59259848.342942.57749869.899930.0026
9902.235919.4033    9999910.191610015.15910.770710046.81919.810210058.01927.3219
10081.81950.9247 10091.2954.550810102.26955.452110113.33969.258210124.39988.2059
10128.57   993.210157.581019.71910179.711036.85110201.841050.344 10212.91059.623
10224.221074.32510235.551083.63310269.541102.00210285.111106.97510314.851111.115
 10372.61111.48210407.791100.38110419.721095.11210431.661086.63210440.981083.415
#Mann= 3 , 0 , 0
9591.507    0.12       09591.507    0.12       010440.98    0.12       0
#XS Ineff= 2 , 0
       0                               0
Bank Sta=9591.507,10440.98
Exp/Cntr=0.3,0.1

Type RM Length L Ch R = 1 ,46817.73,247.787800,247.787800,247.787800
XS GIS Cut Line= 6
512749.925871037800650.254348512512784.977079158800688.207403837
 512843.16935083800757.172040113512951.111970152800897.545715226
513096.603952318 801076.52399972513243.128500893 801263.20609371
#Sta/Elev= 30
9584.471955.40199590.931955.62369618.155950.09529684.274942.09019799.318943.0168
9824.547 941.9349844.206937.24289862.391926.76769875.006922.35249938.826916.6137
  9964.6916.41449977.486909.658710004.65908.376310020.51908.651710029.09 910.378
10041.97916.589310054.85925.094110083.97955.031310093.49960.993810106.38957.6298
 10170.3950.419610180.09948.703510183.01946.572710196.29943.237110221.15944.9322
10228.68947.635210246.58965.227910284.71980.973410310.14985.880410371.421010.588
#Mann= 3 , 0 , 0
9584.471    0.12       09584.471    0.12       010371.42    0.12       0
#XS Ineff= 2 , 0
       0                               0
Bank Sta=9584.471,10371.42
Exp/Cntr=0.3,0.1

Type RM Length L Ch R = 1 ,46569.94,247.787900,247.787900,247.787900
XS GIS Cut Line= 6
512701.696229786800678.144693186512745.302855506800759.890538731
 512777.34841469800857.964343187512787.222052314800954.774365461
512782.271481857 801149.18068318512828.732480013801389.631998399
#Sta/Elev= 30
9633.736944.22179731.977940.99019816.412941.30319867.313938.91119897.412933.5316
9917.443923.42069937.476920.16869977.544 918.7749997.578909.1269 10007.6908.3873
10057.69908.4586 10077.7914.132910107.72936.233310117.72 950.12910127.76960.8869
10137.83975.576710147.89983.531810157.95985.064510168.02991.617810178.121003.106
10198.381018.579 10208.51020.28910218.631031.11510249.231059.82410269.641076.275
 10290.11089.12510300.391094.12610353.131118.46710362.331122.37210367.141122.616
#Mann= 3 , 0 , 0
9633.736  0.1007       09633.736  0.1007       010367.14  0.1007       0
#XS Ineff= 2 , 0
       0                               0
Bank Sta=9633.736,10367.14
Exp/Cntr=0.3,0.1

Type RM Length L Ch R = 1 ,46322.16,247.787800,247.787800,247.787800
XS GIS Cut Line= 6
512494.100750891 800689.91557085512513.738992095800776.199917486
512531.565363779800907.697930704512539.895353256801113.829371798
512551.034273877801258.135927666512579.167629538801465.770427362
#Sta/Elev= 30
 9637.85950.32489663.823945.06679674.107940.5826 9846.32938.78679916.605934.3222
 9926.64930.8399 9946.66919.73229956.669917.03969966.678917.20159986.683907.1448
9996.683 906.70510016.69910.438110076.73910.176610106.82914.645610116.84920.5355
10126.87933.2255 10136.9943.327210197.08990.648710207.111000.48810217.171001.044
10227.251006.14710237.33 1023.43 10247.41037.55210267.55 1052.1910297.78 1064.14
10317.931069.03710338.091067.86710368.381074.80510408.911092.83810419.821093.599
#Mann= 3 , 0 , 0
 9637.85  0.0528       0 9637.85  0.0528       010419.82  0.0528       0
#XS Ineff= 2 , 0
       0                               0
Bank Sta=9637.85,10419.82
Exp/Cntr=0.3,0.1

Type RM Length L Ch R = 1 ,46074.37,247.787800,247.787800,247.787800
XS GIS Cut Line= 6
512278.392911466800702.146427722 512282.88485844800758.468338858
512287.165495699800853.433693644512295.211408872801242.548230419
512298.704563428801349.329145588512306.595321745801470.488256719
#Sta/Elev= 30
9642.604968.59579685.593965.49219755.693940.56279845.743937.21849905.756931.4168
 9925.76924.46289935.762918.23929965.769915.44719985.773904.81549995.775 904.029
10065.79910.7662 10095.8915.6289 10115.8920.8073 10125.8925.433110135.81936.8092
10155.81953.115810185.82968.244210215.83990.332810225.84995.552310235.84 1006.14
10245.851009.61610255.851009.81810265.861013.41610285.871027.04210305.911028.556
10345.99 1043.2210376.051060.10110386.081069.986 10396.11074.30110411.621073.891
#Mann= 3 , 0 , 0
9642.604   0.048       09642.604   0.048       010411.62   0.048       0
#XS Ineff= 2 , 0
       0                               0
Bank Sta=9642.604,10411.62
Exp/Cntr=0.3,0.1

Type RM Length L Ch R = 1 ,45826.58,247.787900,247.787900,247.787900
XS GIS Cut Line= 6
512064.915714577800714.253090154512061.353330703800800.913933722
512043.986029546801048.155899173512032.352007012801218.145450024
512025.342275626801346.770818167512024.172055981 801411.23862054
#Sta/Elev= 30
9664.415951.63439715.205952.4972 9745.23944.8777 9765.27944.55199775.294940.0892
9795.344935.45699905.615921.76389925.664914.27229965.762911.47979975.787904.5991
9985.812901.891910005.86901.825210015.88902.743210025.91 907.66210035.93906.9407
10045.95908.315510096.07920.917710126.14944.221810176.25972.619910186.27972.5051
10196.28976.7615 10206.3983.484110236.34995.772110246.361001.662 10276.41024.573
10286.421030.69410296.431031.14810306.431034.52210316.44 1035.8710362.681038.385
#Mann= 3 , 0 , 0
9664.415  0.0523       09664.415  0.0523       010362.68  0.0523       0
#XS Ineff= 2 , 0
       0                               0
Bank Sta=9664.415,10362.68
Exp/Cntr=0.3,0.1

Type RM Length L Ch R = 1 ,45578.79,495.575700,495.575700,495.575700
XS GIS Cut Line= 6
511859.765894263800658.469627201 511843.69050269800771.450462952
511819.101395702800912.053811867511771.984019956801154.457796896
511746.369655186801312.213983062511741.756825158801351.990670021
#Sta/Elev= 30
 9637.03939.19679670.863 938.1529704.231934.35849825.815930.54169835.967929.0957
9846.118924.4171 9856.27923.19739886.726923.53589896.889921.07779907.081915.5817
9917.273912.87079958.042910.55179988.618902.2468   10009901.164410019.18903.1711
10029.36908.242610059.91913.2227 10070.1922.124110080.28933.500710110.83960.8564
10151.51990.299710161.641001.284 10181.91012.46610192.031015.26610222.42 1013.51
10242.691027.40310252.821032.34510262.951034.91910312.541037.52410340.691036.567
#Mann= 3 , 0 , 0
 9637.03  0.0448       0 9637.03  0.0448       010340.69  0.0448       0
#XS Ineff= 2 , 0
       0                               0
Bank Sta=9637.03,10340.69
Exp/Cntr=0.3,0.1

Type RM Length L Ch R = 1 ,45083.22,394.581600,394.581600,394.581600
XS GIS Cut Line= 6
511467.822574992800324.486258401511453.793914223800424.531905156
 511418.02526777   800588.873023511236.920955085801126.575547276
511202.892373569 801248.42856157511171.084211638801413.881372097
#Sta/Elev= 30
 9436.851013.2859457.5241010.5319477.731996.49649508.043986.79219518.147969.1375
9538.358966.28939568.904946.1019 9599.45937.61289609.633932.25259619.872932.1174
9630.154926.84119640.436927.91089661.001922.95549681.566922.26129858.816922.1149
9922.398908.34359954.192907.68269975.388900.378110028.46900.869610039.08907.4188
10070.96911.098610092.22924.366510155.98944.0048 10166.6945.121210229.84 945.716
10261.44948.842610488.77951.022610519.25944.912610549.63943.736610568.71937.9647
#Mann= 3 , 0 , 0
 9436.85  0.0527       0 9436.85  0.0527       010568.71  0.0527       0
#XS Ineff= 2 , 0
       0                               0
Bank Sta=9436.85,10568.71
Exp/Cntr=0.3,0.1

Type RM Length L Ch R = 1 ,44688.64,576.704800,576.704800,576.704800
XS GIS Cut Line= 4
510983.960837394800380.824323773510932.739085586801113.710874914
510910.721070392801231.779017492510901.572407863801301.259080647
#Sta/Elev= 30
9638.5331056.1689662.7681054.2019692.8411038.3689742.9631017.2979763.0121003.692
9773.0361000.2199783.061991.17869803.109978.01099813.134973.39779823.158965.9466
9843.207947.01079893.329 921.0359933.427910.78869953.475910.1452  9963.5906.9354
9973.524900.80899983.548898.8245 10003.6898.361810023.65898.476310063.74904.8661
10103.84907.564310113.87910.012810123.89914.819610143.94917.367210264.23927.4294
10425.38929.402610435.55929.958610445.73932.802910466.07931.133610563.39931.2532
#Mann= 3 , 0 , 0
9638.533    0.04       09638.533    0.04       010563.39    0.04       0
#XS Ineff= 2 , 0
       0                               0
Bank Sta=9638.533,10563.39
Exp/Cntr=0.3,0.1

Type RM Length L Ch R = 1 ,44111.93,267.652800,267.652800,267.652800
XS GIS Cut Line= 6
510402.935903796800447.182480893510398.761166168800638.699460825
510370.510972031 800809.15888072 510361.46707228800926.735403278
510363.065487532801051.743274414 510384.93310303801226.768617463
#Sta/Elev= 30
9734.7911006.6719752.626999.04389782.629997.60439802.632991.95339812.634 985.114
9867.296958.80829882.691946.74939902.746 926.8899912.774 921.3199922.801919.3436
9963.143903.03029993.575895.261710013.93895.4551 10034.3901.154810074.91906.0796
10085.02904.437410105.22907.454910125.32906.739810255.57913.684110275.57922.9673
10305.58951.119110315.59956.4381 10325.6955.5528 10335.6958.990610345.62970.9796
10355.65979.423810446.181016.90310456.281019.53510486.571020.41110518.861013.805
#Mann= 3 , 0 , 0
9734.791  0.0453       09734.791  0.0453       010518.86  0.0453       0
#XS Ineff= 2 , 0
       0                               0
Bank Sta=9734.791,10518.86
Exp/Cntr=0.3,0.1

Type RM Length L Ch R = 1 ,43844.28,247.787800,247.787800,247.787800
XS GIS Cut Line= 6
510057.454928761800442.612438172510129.020533427800746.239144639
510187.682879815801019.103549576510213.060920382801115.065237413
510238.459779844801194.944731911510255.357112577801238.790614507
#Sta/Elev= 30
9709.8411055.5529722.6691048.0839743.2321032.9929763.7751014.5059774.047  1002.8
9784.318998.3313 9794.59 999.1849815.133998.25269825.405 994.4639856.219967.5724
 9928.12913.07089948.663904.32979958.934898.34159969.206894.97129989.749894.4912
10020.53 895.49410030.76899.525810040.99899.844910061.44903.677210071.67902.8997
10102.36 906.16310143.27905.4399 10153.5907.229810276.24911.605310306.99914.3273
10369.06933.244610400.09937.211510439.56945.891110516.19 971.00510530.97  974.75
#Mann= 3 , 0 , 0
9709.841  0.0415       09709.841  0.0415       010530.97  0.0415       0
#XS Ineff= 2 , 0
       0                               0
Bank Sta=9709.841,10530.97
Exp/Cntr=0.3,0.1

Type RM Length L Ch R = 1 ,43596.49,247.787900,247.787900,247.787900
XS GIS Cut Line= 6
509760.731230309800560.627545515509854.222333004 800739.05545037
509910.277786325800834.871038716510047.089396224801089.852381719
510123.075157752 801222.76163621510162.257613328801285.340364131
#Sta/Elev= 30
9729.0711053.3689767.8761034.1329801.744 1023.289835.6131007.5069846.903998.5169
9869.482971.88839889.091954.14579903.351939.5238 9925.93930.26039937.372 923.099
9960.466905.60689972.064894.9488 9983.56889.809310018.39 891.47410051.51895.9663
10064.36894.334710075.71895.472810087.06902.126510098.41904.665510268.64 911.046
10279.99909.490210348.33928.123410382.89932.947710394.41932.066410405.93938.0693
10417.45940.720810498.42956.066210522.02962.725110533.82962.128710557.82967.3324
#Mann= 3 , 0 , 0
9729.071    0.04       09729.071    0.04       010557.82    0.04       0
#XS Ineff= 2 , 0
       0                               0
Bank Sta=9729.071,10557.82
Exp/Cntr=0.3,0.1

Type RM Length L Ch R = 1 , 43348.7,247.787800,247.787800,247.787800
XS GIS Cut Line= 6
509498.540225715800728.311828804509573.678729214 800817.87604996
509692.218588196800948.860594712509697.005335632800953.938661166
509972.531589298801242.772853136510063.229714008801334.854313782
#Sta/Elev= 30
9700.4541090.9389726.0631069.098 9735.291065.3429741.6221063.7839761.3961067.402
9803.8591055.3719819.3311047.0149834.2341035.1689878.943 994.0519908.749970.3772
9938.555942.14579953.458925.54949968.361901.97969975.328895.39099988.815888.7156
10027.07888.438810071.57903.0028   10114906.886510223.59 909.48510265.05916.3869
10302.34925.291210320.33927.946710334.15927.011410360.29938.854110375.61942.9823
10417.94950.915510445.41958.803310473.48962.862210503.44  977.7210529.42986.9747
#Mann= 3 , 0 , 0
9700.454  0.0639       09700.454  0.0639       010529.42  0.0639       0
#XS Ineff= 2 , 0
       0                               0
Bank Sta=9700.454,10529.42
Exp/Cntr=0.3,0.1

Type RM Length L Ch R = 1 ,43100.91,247.787900,247.787900,247.787900
XS GIS Cut Line= 6
509309.647504959800959.542573179509470.255572477801090.243514474
509659.537530255801229.093527677509724.708797241801272.969389056
509821.945698937801334.419883343509932.100666713801400.418837395
#Sta/Elev= 30
9728.4441088.864 9748.481083.4739768.0631070.0159815.5381041.5499864.582989.5102
9903.097945.31479928.774 909.9029941.442898.66199953.921893.34169978.881888.9822
10016.13886.759710028.51887.777910044.54893.486710078.02900.628810152.28904.4176
10188.91911.194310237.13913.261610248.84916.269510284.67933.113810308.33950.3253
10320.16954.100810331.99965.849910343.82974.053510367.43990.2447 10402.41010.871
10423.361010.68210437.371017.99210472.341023.004   104841021.81410492.281022.774
#Mann= 3 , 0 , 0
9728.444    0.12       09728.444    0.12       010492.28    0.12       0
#XS Ineff= 2 , 0
       0                               0
Bank Sta=9728.444,10492.28
Exp/Cntr=0.3,0.1

Type RM Length L Ch R = 1 ,42853.13,247.787800,247.787800,247.787800
XS GIS Cut Line= 6
509142.165493399801229.775263361509168.313449599801243.682366134
509273.001616025 801293.09122047509385.241371472801337.957583742
509406.620475648801345.870463453509818.139184852801488.381250953
#Sta/Elev= 30
 9711.951028.261 9748.961010.7859768.0831005.4999782.1341005.1759793.192 1008.21
9826.3651010.9119859.481981.42559902.558 932.9419924.097916.50199943.294896.3826
9977.944887.1518 9988.61886.192810020.45888.830310031.03892.723610041.62891.9038
10062.78898.078410094.53902.136210136.86911.878610179.19912.628410189.77913.7872
10200.36917.594210210.94924.486810221.52926.677710242.69938.999710253.27942.6972
10285.02963.4312 10295.6 967.75510327.35973.738910369.68999.6486 10436.51052.013
#Mann= 3 , 0 , 0
 9711.95    0.12       0 9711.95    0.12       0 10436.5    0.12       0
#XS Ineff= 2 , 0
       0                               0
Bank Sta=9711.95,10436.5
Exp/Cntr=0.3,0.1

Type RM Length L Ch R = 1 ,42605.34,247.787900,247.787900,247.787900
XS GIS Cut Line= 6
509061.051212996801503.535959671509219.156145975801553.315376577
509315.133103005801578.482438323 509409.52151387801599.352352428
509560.742325833801625.759071639509757.533486299 801652.16093638
#Sta/Elev= 30
9711.1191019.0469778.622980.23339799.498980.68319830.812963.25469851.689960.1715
9872.565940.27119882.944922.09269913.958897.18079934.635892.11999955.311890.7522
9976.125884.327410037.46 886.26710057.93 890.91510078.37904.737610098.73908.3475
10108.91916.431710129.27938.428810149.59951.597110159.72961.377210169.85 967.416
10179.98977.787410200.24974.945810210.37985.1788 10220.5991.992510270.97 1013.24
10301.241018.49110311.331023.62810321.421025.23110371.871012.74610424.871050.898
#Mann= 3 , 0 , 0
9711.119    0.12       09711.119    0.12       010424.87    0.12       0
#XS Ineff= 2 , 0
       0                               0
Bank Sta=9711.119,10424.87
Exp/Cntr=0.3,0.1

Type RM Length L Ch R = 1 ,42357.55,247.787800,247.787800,247.787800
XS GIS Cut Line= 6
508981.142411707801786.918592283509075.695616655801807.321085796
509142.958967283801817.810158618509209.739293465801824.800442358
509303.321259922801828.017528219 509693.24794252801825.884965408
#Sta/Elev= 30
9673.3691023.0539749.019986.90889759.217980.21899789.662 970.6099809.904955.4017
9820.025944.74219840.253933.06749860.362914.96729880.472902.29359890.526898.1511
9910.613893.736310010.68882.421810030.68883.163510040.68  885.4910090.68 904.689
10100.68904.808710120.68916.058210130.68918.488310170.68946.895710180.68951.5561
10210.68977.993710220.68979.646310250.681007.08510300.681041.30810310.681047.183
10330.681044.95310340.681046.91410360.681070.41210370.681077.24210388.941085.425
#Mann= 3 , 0 , 0
9673.369  0.0553       09673.369  0.0553       010388.94  0.0553       0
#XS Ineff= 2 , 0
       0                               0
Bank Sta=9673.369,10388.94
Exp/Cntr=0.3,0.1

Type RM Length L Ch R = 1 ,42109.76,247.787900,247.787900,247.787900
XS GIS Cut Line= 6
508920.765424573802024.189559293509052.599391587802049.579166969
509189.541415883802068.920954148 509278.61408838802075.554886154
509459.672959412802075.949304112509603.555560021802068.267951492
#Sta/Elev= 30
9611.9471006.7549626.487998.8595 9657.13995.50399664.999992.77989677.539984.7172
9708.017970.39519738.496962.51889748.641957.0623 9758.74954.41419799.137935.9169
9809.236932.82819819.336 923.4569829.435916.98559849.633900.28489930.102890.6227
9950.157886.48239960.185885.90579970.213881.78219980.223880.000610000.22879.6095
10020.22879.899710080.22901.704810100.22918.262710130.22936.118610160.23943.4159
10180.24955.363410200.25961.158410210.26966.145710230.27979.376910299.031016.322
#Mann= 3 , 0 , 0
9611.947   0.055       09611.947   0.055       010299.03   0.055       0
#XS Ineff= 2 , 0
       0                               0
Bank Sta=9611.947,10299.03
Exp/Cntr=0.3,0.1

Type RM Length L Ch R = 1 ,41861.97,247.787800,247.787800,247.787800
XS GIS Cut Line= 6
508862.419467145802253.478935816509196.737761244802306.428582244
 509297.92555869802325.745819454509339.790322402802330.428875932
509465.548977159802332.406641487509549.669866422 802324.05029107
#Sta/Elev= 30
9596.2991013.4259609.1131004.7819680.158970.62499710.506950.79869720.622948.4419
9730.738951.8604 9750.97944.97489771.202941.98649781.318936.6726 9801.55933.3321
9821.782 925.1159831.898 916.2439862.246902.35119872.362   902.29882.478897.8671
9912.826891.09859943.228890.50839973.772879.2583 10014.5878.876110044.95885.3896
10055.01891.403710075.14895.117310095.19920.467710115.22941.849710165.25982.6288
10175.25 986.06510185.25995.725310195.251001.72810255.421021.92110290.361040.389
#Mann= 3 , 0 , 0
9596.299   0.053       09596.299   0.053       010290.36   0.053       0
#XS Ineff= 2 , 0
       0                               0
Bank Sta=9596.299,10290.36
Exp/Cntr=0.3,0.1

Type RM Length L Ch R = 1 ,41614.19,247.787800,247.787800,247.787800
XS GIS Cut Line= 6
 508819.05948906802567.139154086509021.403728853802573.951719773
509331.682325149802560.636283011509405.415483239802549.193707886
 509488.27115293 802528.55334729509568.557484021802500.907074203
#Sta/Elev= 30
9553.118949.72229579.114 942.4929599.157945.12249621.199  943.699649.219935.6338
9679.236948.34379739.238932.55139769.242926.75649809.252923.73199849.266914.1207
9899.307887.46049929.332885.43619959.357878.59399969.365878.32479989.382882.6619
 9999.39882.042210009.41877.683110019.44877.538410029.47877.924710049.53887.4864
10069.62890.468610099.98921.468110150.75964.859110161.06969.319410191.97 972.653
10212.59983.438310254.45995.294810275.54 1005.7610300.491024.605 10311.21026.832
#Mann= 3 , 0 , 0
9553.118  0.0457       09553.118  0.0457       0 10311.2  0.0457       0
#XS Ineff= 2 , 0
       0                               0
Bank Sta=9553.118,10311.2
Exp/Cntr=0.3,0.1

Type RM Length L Ch R = 1 , 41366.4,247.787900,247.787900,247.787900
XS GIS Cut Line= 6
508929.385682801802919.248623914509066.809250467802894.092825864
509162.223545805802866.501062488509273.840278084802824.827806971
 509428.07818623802751.443927939509608.961678552802635.972079203
#Sta/Elev= 30
9587.4421093.974  9613.3 1091.359623.3951087.8289643.6311072.927 9653.851068.234
9674.2871070.2659684.5061067.8849727.2291042.6299777.3941009.8359787.8041000.572
9808.623988.40519819.033978.66469829.497966.45189840.101958.14249861.118920.8495
9893.182891.18349914.695883.71079925.451877.30289957.853876.20469990.479876.9693
10034.51885.011310079.24889.006410124.61921.200210147.69930.210410159.23937.5965
10218.09960.592410229.92 960.33110241.75962.6237 10280.1981.698510331.321003.017
#Mann= 3 , 0 , 0
9587.442    0.04       09587.442    0.04       010331.32    0.04       0
#XS Ineff= 2 , 0
       0                               0
Bank Sta=9587.442,10331.32
Exp/Cntr=0.3,0.1

Type RM Length L Ch R = 1 ,41118.61,247.787800,247.787800,247.787800
XS GIS Cut Line= 6
509161.673361349803229.495865828509244.068292784803192.230291061
509287.170416953803166.117980693 509386.45657423803086.143371244
509460.256893604  803007.0138776509682.781361037802733.103240357
#Sta/Elev= 30
9618.134 1190.319643.1521152.2099656.4231136.8319676.3281097.3599698.553  1063.3
 9709.72 1062.449744.7951025.865 9760.92 999.9059768.722984.19839777.869971.0331
9793.493 961.2169818.263938.03349858.114906.95649898.798885.97019930.408876.3159
9941.572 876.25410010.39877.6705 10023.2880.656610050.26881.237110061.66884.3703
 10087.3884.750610100.12890.7714 10114.2 893.46310162.15918.407710242.07942.9052
10267.07956.579610293.16959.714510304.54964.542410319.25974.783110347.81981.7554
#Mann= 3 , 0 , 0
9618.134  0.0919       09618.134  0.0919       010347.81  0.0919       0
#XS Ineff= 2 , 0
       0                               0
Bank Sta=9618.134,10347.81
Exp/Cntr=0.3,0.1

Type RM Length L Ch R = 1 ,40870.82,247.787900,247.787900,247.787900
XS GIS Cut Line= 6
509562.039751756803338.503708529509609.014675397803273.585649822
509629.104461877803236.596105889509728.234972617802986.566669457
509771.896451695  802887.8641173509811.310821109802812.751061885
#Sta/Elev= 30
9749.463962.21489767.363951.23769779.974947.22559791.989940.49079816.019931.2754
9828.034925.24089839.504917.56569862.263898.62549873.584892.22299885.909892.3939
9895.607889.82299906.619882.9901 9917.63880.74059934.631878.39289960.831 877.982
9971.573875.01229993.056872.824310025.12873.840510046.48883.045710089.19 886.314
10110.54890.899510121.22894.891810142.61905.760910186.35932.010810231.78949.0468
10255.71960.905410274.45962.819910296.86975.894110308.22979.707310333.67978.4116
#Mann= 3 , 0 , 0
9749.463    0.12       09749.463    0.12       010333.67    0.12       0
#XS Ineff= 2 , 0
       0                               0
Bank Sta=9749.463,10333.67
Exp/Cntr=0.3,0.1

Type RM Length L Ch R = 1 ,40623.04,247.787800,247.787800,247.787800
XS GIS Cut Line= 6
509820.766392916803494.973629311509888.986571223803287.627300218
509926.971075892803144.489991397509961.625932813803032.224549592
509995.173727363802940.678660572510012.732370436802898.699670881
#Sta/Elev= 30
9693.864987.89999714.871981.79949772.105950.77179788.491935.95649809.525911.6857
9820.058907.98189830.597907.60049851.677 893.9039872.756885.38379925.222875.5357
9945.934874.09649966.645877.43249987.357872.936110018.37872.8165 10028.7873.0646
10039.04879.019210049.38  881.8410080.64883.4277 10122.5 891.84710143.43905.6653
 10153.9 909.02610174.83921.727210185.43920.941710196.08928.823110206.73939.6955
10238.68954.650510249.33963.171510270.63963.587210281.39970.791210320.74987.0902
#Mann= 3 , 0 , 0
9693.864   0.089       09693.864   0.089       010320.74   0.089       0
#XS Ineff= 2 , 0
       0                               0
Bank Sta=9693.864,10320.74
Exp/Cntr=0.3,0.1

Type RM Length L Ch R = 1 ,40375.25,247.787900,247.787900,247.787900
XS GIS Cut Line= 6
510059.481670707803601.310434878510146.817188829803285.701686591
510161.384640455803224.561828837510179.464968771803165.723478869
510219.225895047 803060.28708604 510247.39265427 802998.83158353
#Sta/Elev= 30
9641.084980.7976 9668.39 968.6479689.147955.68789699.525940.85469709.903931.9172
9720.282931.8051 9730.66925.83829761.795901.70239772.174895.26519803.309886.9569
9813.687 887.4129855.201877.94579886.336878.69529907.088877.85659961.651872.6943
10010.37872.060710030.96873.780710062.33890.047310083.26 899.09510093.73901.3664
10104.34906.376610114.95 915.76810136.17940.781510146.81947.672710168.32960.5458
10189.84 966.57210211.48974.220310222.48981.404210244.48990.559310273.271009.422
#Mann= 3 , 0 , 0
9641.084  0.0994       09641.084  0.0994       010273.27  0.0994       0
#XS Ineff= 2 , 0
       0                               0
Bank Sta=9641.084,10273.27
Exp/Cntr=0.3,0.1

Type RM Length L Ch R = 1 ,40127.46,247.787800,247.787800,247.787800
XS GIS Cut Line= 6
510235.262920707803666.414601535510310.071365625803482.977886528
 510338.07587108803428.864482403510378.105261326803358.481711969
510480.898062944803190.087327227510527.842811555803118.502497539
#Sta/Elev= 30
9660.993951.9392 9673.32950.3988 9684.12944.62929705.719926.07439716.519919.0257
9781.316889.37329835.314 879.7529856.913878.6192 9868.08880.21469901.859876.8021
9970.344 874.6439993.441867.0301 10016.8867.043310028.51868.463610052.62879.5222
10063.66886.554710075.37896.4069   10091897.572310098.81901.427210110.52901.7606
10122.24907.783710129.39909.859810148.58920.174710157.39926.445710180.82938.4633
10192.53948.719210204.36 953.41110240.18 959.913   10276979.5671 10283.9979.9602
#Mann= 3 , 0 , 0
9660.993   0.048       09660.993   0.048       0 10283.9   0.048       0
#XS Ineff= 2 , 0
       0                               0
Bank Sta=9660.993,10283.9
Exp/Cntr=0.3,0.1

Type RM Length L Ch R = 1 ,39879.67,247.787900,247.787900,247.787900
XS GIS Cut Line= 6
510395.853198469803774.921545982510467.571593046803662.902749211
510492.042274624803618.235028878510541.602874398803544.818952724
510635.513395786  803435.6320979510808.435078979803225.397645116
#Sta/Elev= 30
9661.191942.94349684.846940.16949715.247925.42339756.089901.43469791.711887.6866
9826.017 882.5749848.967 883.431 9887.89  877.899922.495876.7356  9954.5873.0632
9969.987867.50929998.992866.709210016.11867.067910031.33871.076610046.55870.4687
10061.77876.289210065.35878.229810091.44 916.85610104.29928.8807 10108.8931.4824
10140.64941.286710156.56941.513410172.48945.663310194.25958.094810252.08977.5261
   10268985.825410283.92991.441110299.791003.50610314.821010.21110350.041020.387
#Mann= 3 , 0 , 0
9661.191  0.0472       09661.191  0.0472       010350.04  0.0472       0
#XS Ineff= 2 , 0
       0                               0
Bank Sta=9661.191,10350.04
Exp/Cntr=0.3,0.1

Type RM Length L Ch R = 1 ,39631.88,743.363500,743.363500,743.363500
XS GIS Cut Line= 6
 510634.56847626803896.449323773510725.904204041803779.836175755
510792.637528777803624.286814451510841.934005529803535.096148416
510898.785269827803456.731143788 510988.50043273803358.582078382
#Sta/Elev= 30
9681.595918.02999696.139917.74579708.841914.77649746.947 899.7559785.054890.4765
9812.036882.58959823.161 881.0429879.843879.74269921.495874.19239943.416867.1601
9976.297866.347210020.66867.379410031.92868.997410054.45882.183710077.76901.0337
10089.42914.253410101.08923.048210106.37926.438710113.22928.938910137.51945.3656
 10154.4953.607110174.73968.407810191.62970.262610200.08975.110910213.22977.7124
10238.25975.470710268.13977.403910282.67987.091910297.21993.188210330.851013.836
#Mann= 3 , 0 , 0
9681.595  0.0948       09681.595  0.0948       010330.85  0.0948       0
#XS Ineff= 2 , 0
       0                               0
Bank Sta=9681.595,10330.85
Exp/Cntr=0.3,0.1

Type RM Length L Ch R = 1 ,38888.52,743.363500,743.363500,743.363500
XS GIS Cut Line= 6
510669.290698469803898.619462669510821.200420707 803981.08474043
 511111.86557957804202.588179725511201.319215485804210.622003081
511240.727110346804220.160065191511422.654578894804289.341397841
#Sta/Elev= 30
9416.167914.93929471.462906.46429513.691 897.1339555.303890.46179644.085887.4381
 9669.23884.90999719.521882.92859760.461879.36119820.103871.17049870.394870.7112
9908.946863.17599920.685863.27369933.257869.0812 9945.83869.92679957.644 867.808
9967.797862.77839977.949 860.9059997.955860.772710017.97860.900510038.14864.7847
10068.87878.387310079.16887.177210100.04898.911310110.55907.168510163.48952.6106
10206.39993.535710217.221002.15310249.691023.61510271.431034.04510279.821035.378
#Mann= 3 , 0 , 0
9416.167   0.095       09416.167   0.095       010279.82   0.095       0
#XS Ineff= 2 , 0
       0                               0
Bank Sta=9416.167,10279.82
Exp/Cntr=0.3,0.1

Type RM Length L Ch R = 1 ,38145.16,247.787900,247.787900,247.787900
XS GIS Cut Line= 6
510658.440004021803924.661129296510593.088977128804055.348830119
510527.005937189804155.712455168510465.695760787 804267.94678013
510417.090734065804402.748243868510396.841493845804505.953470185
#Sta/Elev= 30
9627.582909.34869661.502894.05999672.683889.55679683.864886.52889706.225884.4565
9750.947884.61599787.877881.51679805.405878.55039822.932871.7869 9834.02868.8671
9869.441866.36189881.248866.57529915.935862.50689938.788862.60079961.641855.6621
9984.494854.4982 9995.92855.016910007.24857.064110029.47868.662610040.35881.4597
10051.23890.873810072.93901.559110094.17914.673610104.79918.244410136.32 923.331
10174.29938.815510208.69956.884910218.86963.546910228.99966.587110270.49990.6858
#Mann= 3 , 0 , 0
9627.582    0.12       09627.582    0.12       010270.49    0.12       0
#XS Ineff= 2 , 0
       0                               0
Bank Sta=9627.582,10270.49
Exp/Cntr=0.3,0.1

Type RM Length L Ch R = 1 ,37897.37,247.787800,247.787800,247.787800
XS GIS Cut Line= 6
510460.205959772803866.945186696510404.037186009803914.705077323
510364.299699934803961.800921959510293.498232545804066.975351735
510196.117433898804279.737753336510153.446037295804453.016034165
#Sta/Elev= 30
9677.246903.08789695.477895.63359722.457888.23159751.587 882.7689816.777878.7144
9829.141876.76149866.234866.46289878.295865.03159913.726863.37979925.536864.8959
9937.346864.40219948.729866.32359982.565856.01129993.844854.407910015.98854.1457
10026.98854.739710037.98861.000310059.98864.202610070.98869.069910081.98876.5866
10092.99881.5374 10125.7 902.45310136.46906.017910168.73910.317310231.85926.1643
10283.46945.4898 10314.2962.554910324.31965.041610344.53973.998910352.64976.2692
#Mann= 3 , 0 , 0
9677.246    0.12       09677.246    0.12       010352.64    0.12       0
#XS Ineff= 2 , 0
       0                               0
Bank Sta=9677.246,10352.64
Exp/Cntr=0.3,0.1

Type RM Length L Ch R = 1 ,37649.58,247.787900,247.787900,247.787900
XS GIS Cut Line= 6
510172.437293365803785.849981101 510073.35425952803951.039907629
 509996.95384644804120.513117251509974.669461919804187.905036068
509955.920610419804267.907854975509943.395673167804395.842562271
#Sta/Elev= 30
 9746.95939.51169793.525907.17829805.366901.16049817.207891.42789829.047887.7146
9840.888  886.579845.113885.14059852.487882.06299863.952873.70339875.418871.6033
9886.883865.54169895.415862.55739921.278863.80639939.668861.3738 9944.11860.2413
9958.106853.698810010.94853.110810052.23860.441110087.23865.159610125.66873.5794
10151.45880.927110172.51884.492110203.98891.626710245.21897.254610275.86904.9385
10326.33914.564810356.58926.671910376.62929.716810396.64934.260510407.49937.7567
#Mann= 3 , 0 , 0
 9746.95    0.12       0 9746.95    0.12       010407.49    0.12       0
#XS Ineff= 2 , 0
       0                               0
Bank Sta=9746.95,10407.49
Exp/Cntr=0.3,0.1

Type RM Length L Ch R = 1 ,37401.79,247.787800,247.787800,247.787800
XS GIS Cut Line= 6
509903.229189688 803705.13921195509787.668030183803985.351039805
509768.368468169804065.383637251509763.557509537 804220.49604713
509780.651595107804345.281256587509802.226919718804441.552139844
#Sta/Elev= 30
 9784.62939.15759805.771 917.1949827.069907.04079837.719 897.4879880.905863.1622
9891.732861.11299903.442861.51469957.415857.42599964.312856.55239979.362851.9473
 10001.3851.079310023.13851.835510044.65855.550610076.77858.385310129.08866.1451
10169.86877.147510280.22877.393410330.26880.179610340.32881.676810360.44887.1509
10390.65899.539310410.91904.526810451.45922.760310482.12934.248310492.35936.9479
10502.58938.3155 10512.8937.347810523.03933.641910543.65933.057410550.41931.1534
#Mann= 3 , 0 , 0
 9784.62    0.12       0 9784.62    0.12       010550.41    0.12       0
#XS Ineff= 2 , 0
       0                               0
Bank Sta=9784.62,10550.41
Exp/Cntr=0.3,0.1

Type RM Length L Ch R = 1 ,37154.01,247.787800,247.787800,247.787800
XS GIS Cut Line= 6
509506.080358561803730.004439649509617.705658261803904.316658232
509638.261353059803946.092954263509653.596698453803999.278276906
509693.622583776804190.964656776509774.831158618804467.767049177
#Sta/Elev= 30
9819.142949.46729860.566930.73269907.634 900.9459919.401 884.0019930.326872.4233
9942.975862.72139991.172849.742310015.08 848.97210026.94849.7502 10060.7856.4275
10092.45858.328910133.97865.840910154.41866.288710174.84869.104610195.27873.7653
10205.48874.650110246.35875.343610348.82874.333310379.86875.6562 10410.9879.0063
10441.94884.871110462.85895.077910483.81900.280810494.29907.066910515.26916.4673
10525.74919.825510536.22921.1013 10546.7920.111610579.68912.116510612.49907.1528
#Mann= 3 , 0 , 0
9819.142    0.12       09819.142    0.12       010612.49    0.12       0
#XS Ineff= 2 , 0
       0                               0
Bank Sta=9819.142,10612.49
Exp/Cntr=0.3,0.1

Type RM Length L Ch R = 1 ,36906.22,247.787900,247.787900,247.787900
XS GIS Cut Line= 6
509285.907647438803947.642484466509473.777158901804076.912794456
509559.708607847 804168.61643704509628.246903623804271.493729447
509673.466696906 804355.92394126509740.205118885804500.900587203
#Sta/Elev= 30
9851.762948.44069862.754939.29529874.844930.76829900.444 907.9419918.239889.8582
9923.202885.55589936.033877.66329954.156864.25489971.108852.95359982.984849.7794
10018.68849.109410030.74849.806310056.12854.401810081.65 856.78310095.55856.4312
10123.36862.283710137.27862.336610174.72867.981510310.09872.113110344.77873.7364
10390.15877.5499 10435.3  883.7810451.86889.337110479.68894.743210498.15895.2773
10512.73897.355410523.67895.484810545.56904.880310567.45 912.17610584.85 916.475
#Mann= 3 , 0 , 0
9851.762    0.12       09851.762    0.12       010584.85    0.12       0
#XS Ineff= 2 , 0
       0                               0
Bank Sta=9851.762,10584.85
Exp/Cntr=0.3,0.1

Type RM Length L Ch R = 1 ,36658.43,247.787800,247.787800,247.787800
XS GIS Cut Line= 6
508937.432646125804088.354253101509083.363049529804165.623413072
509350.221210405804270.003482713509447.172060065804321.632025806
509568.534326411804423.236347962509674.699586205804563.582605554
#Sta/Elev= 30
9608.439964.32569629.139953.52899663.547944.71899726.296 921.0339775.471908.6508
9786.364908.37199797.257910.7772 9808.15908.96999822.553902.40359845.109887.9019
9875.255870.72479883.882866.43829894.631863.22869905.379863.13979937.417858.1214
9948.038852.86589958.659850.9216 9969.28 852.322 10054.7847.497210076.75854.4082
10117.57858.141110132.97 862.61110144.56864.327810331.24872.499210384.03877.1723
10409.56885.207110434.42901.666610458.63913.507310470.74917.622610505.14924.1818
#Mann= 3 , 0 , 0
9608.439    0.12       09608.439    0.12       010505.14    0.12       0
#XS Ineff= 2 , 0
       0                               0
Bank Sta=9608.439,10505.14
Exp/Cntr=0.3,0.1

Type RM Length L Ch R = 1 ,36410.64,247.787900,247.787900,247.787900
XS GIS Cut Line= 6
508828.541701214804274.458777147508910.928082288804341.741872139
509001.166879573804394.440127361509372.551630505804560.190322286
509496.016029947804653.765830435509599.997670934804767.484275375
#Sta/Elev= 30
9562.672912.55539571.428910.36839584.985909.51099599.881905.24419641.632898.1674
9685.729892.91319744.001878.53649766.693875.88399799.977866.47989822.036862.4799
9854.927861.41499887.364854.29999941.196849.53989973.286846.982410005.39846.7995
10026.85852.553810048.67853.052210070.57859.016610137.46867.527210232.38877.4436
10282.54878.859510295.58882.772810306.76888.718410348.63915.763810366.25928.6354
10380.49931.561610408.41928.007310448.24918.029210474.12915.622410490.27911.0352
#Mann= 3 , 0 , 0
9562.672    0.12       09562.672    0.12       010490.27    0.12       0
#XS Ineff= 2 , 0
       0                               0
Bank Sta=9562.672,10490.27
Exp/Cntr=0.3,0.1

Type RM Length L Ch R = 1 ,36162.85,495.575700,495.575700,495.575700
XS GIS Cut Line= 6
508767.247997862804379.215288344 508835.62652178804498.896583255
508888.690712818 804561.32905831508984.422933865804634.423168591
509214.743547046804776.204371467509418.833146865804954.837400644
#Sta/Elev= 30
9531.232901.1082 9599.93886.92179668.005881.03679702.099 871.0939730.851866.5286
9759.476865.26319772.591867.92059787.787863.4708 9837.33861.6619 9884.13853.7173
9930.702849.64559942.345846.06489965.631848.0294    9999844.695810035.61 845.934
10059.17853.837310094.93856.601610142.64867.943810155.09868.577310167.55872.5066
10190.61875.459610204.92874.003810242.84 875.65610256.09 880.39510282.59893.9038
10295.83897.556510309.08903.920110322.43908.005910379.41916.842210414.18934.0787
#Mann= 3 , 0 , 0
9531.232    0.12       09531.232    0.12       010414.18    0.12       0
#XS Ineff= 2 , 0
       0                               0
Bank Sta=9531.232,10414.18
Exp/Cntr=0.3,0.1

Type RM Length L Ch R = 1 ,35667.28,300.528000,300.528000,300.528000
XS GIS Cut Line= 6
508745.016870368 804401.29619645508818.219646757 804701.79296797
508830.685999586804859.173051445508825.382592571804923.840325102
508766.904766843 805190.50399335508759.622082122 805365.43940789
#Sta/Elev= 30
 9326.51889.18829372.521880.52169537.658865.56829598.712862.17369619.063862.7915
9659.545 860.0869669.626860.94159689.786858.28419780.008855.69799790.009853.5956
 9810.03852.67289830.058848.98679870.471846.1057 9901.12 847.8479942.409847.8616
9963.053841.08169983.773838.847410015.13839.142210025.43 841.97810035.66  848.02
10045.89856.095910056.12866.373310066.26874.047710086.48887.541310157.05917.9933
10197.19918.696210227.22922.385510247.23 919.84110267.24919.560610307.68926.2869
#Mann= 3 , 0 , 0
 9326.51    0.12       0 9326.51    0.12       010307.68    0.12       0
#XS Ineff= 2 , 0
       0                               0
Bank Sta=9326.51,10307.68
Exp/Cntr=0.3,0.1

Type RM Length L Ch R = 1 ,35366.75,195.047700,195.047700,195.047700
XS GIS Cut Line= 6
508689.127422071804376.035451771508728.719251056804554.891713278
508718.452375515804697.030414281508678.849159247804767.397189554
508465.965799068805002.405503531508376.803626303805179.713460524
#Sta/Elev= 30
9500.683894.6805 9531.01889.21649562.001886.1616 9623.38886.12129664.051882.7282
9684.235878.60969724.297865.93839734.313 864.7499898.335857.72929932.188 852.058
9958.751850.4536 9975.09846.13689989.418839.161710018.03838.6375 10089.2843.1856
10112.07848.184910139.27864.1318 10147.8871.173410157.46882.1681 10195.4919.6421
10216.77937.724710229.28 945.89810241.19948.876210246.39952.000510288.37982.3195
 10305.3996.399810310.95998.874610374.691009.273 10409.71018.43510425.311020.654
#Mann= 3 , 0 , 0
9500.683    0.12       09500.683    0.12       010425.31    0.12       0
#XS Ineff= 2 , 0
       0                               0
Bank Sta=9500.683,10425.31
Exp/Cntr=0.3,0.1

Type RM Length L Ch R = 1 , 35171.7,247.787800,247.787800,247.787800
XS GIS Cut Line= 6
508617.185431516 804371.58099357508579.821796057804523.680622172
508508.663482713804650.987967192508344.648451585804897.633834581
508284.914713213805028.099381269508255.753706303805121.001110998
#Sta/Elev= 30
9616.814914.72519650.455906.29199670.704903.67699701.484895.40169732.873889.1868
9820.324877.5902 9842.66 877.4729866.053873.23619877.824868.50999889.595868.5326
9949.442849.53539961.626848.34359985.995838.00669998.179837.787510083.33842.3119
10095.88844.790610131.93844.613910143.77847.986210178.63866.555810196.22 885.807
10213.49901.437510247.24926.825510280.87948.4132 10313.4959.629210335.08964.0445
10377.95966.4189 10391.4969.495210430.55968.842610451.32971.744510457.53974.0874
#Mann= 3 , 0 , 0
9616.814  0.0544       09616.814  0.0544       010457.53  0.0544       0
#XS Ineff= 2 , 0
       0                               0
Bank Sta=9616.814,10457.53
Exp/Cntr=0.3,0.1

Type RM Length L Ch R = 1 ,34923.92,247.787800,247.787800,247.787800
XS GIS Cut Line= 6
508340.790890475804307.331385331508313.087598283804408.507528955
508186.422647338804762.645549319508162.228305329804837.387881923
508135.610424134 804943.93110299508118.938077992805054.912205799
#Sta/Elev= 30
9689.243914.69789728.199901.4389 9759.36888.90569811.586877.36699864.402874.4807
 9896.18866.0426 9928.09860.61519970.637844.88899981.274837.11889991.911834.1226
10002.55833.877810023.83835.478910055.75841.355710077.03843.129210115.91842.0211
10130.23843.626110172.76864.448910193.78880.621310207.38893.935510225.32906.2686
10246.34913.544110277.49916.524210349.53916.869510359.78913.281910369.93905.8839
10380.07901.396710400.37896.615410430.78 893.13310460.98895.298510470.96891.8834
#Mann= 3 , 0 , 0
9689.243  0.0463       09689.243  0.0463       010470.96  0.0463       0
#XS Ineff= 2 , 0
       0                               0
Bank Sta=9689.243,10470.96
Exp/Cntr=0.3,0.1
