HEC-RAS study 5238_ras.prj: 5238

--- 5238_ras.g01 (geometry) --- (continued)

Type RM Length L Ch R = 1 ,34676.13,247.787900,247.787900,247.787900
XS GIS Cut Line= 6
508071.259990199 804244.67727254508032.817286354804437.038246246
507991.190308188804593.130862221507971.273303372804712.334052768
 507969.67330553804855.868969799507982.049472452804988.788048912
#Sta/Elev= 30
 9708.49895.64859759.518878.40799810.494 866.8449861.678860.45729902.624859.6235
9933.663856.17669944.017853.27079964.725844.10529975.079836.13169985.433832.5964
   10001832.586710006.15 832.59210037.17839.560910078.35841.011210129.29845.7956
10169.72854.1914 10179.8860.802410189.86869.307610199.88870.974910239.95 871.216
10259.95867.509410299.97867.880510329.98870.013210340.02869.627210360.09866.3745
10380.16 871.18310410.27875.384910420.31878.472110430.35882.318610464.36899.2246
#Mann= 3 , 0 , 0
 9708.49  0.0507       0 9708.49  0.0507       010464.36  0.0507       0
#XS Ineff= 2 , 0
       0                               0
Bank Sta=9708.49,10464.36
Exp/Cntr=0.3,0.1

Type RM Length L Ch R = 1 ,34428.34,247.787800,247.787800,247.787800
XS GIS Cut Line= 6
507729.842891177 804183.00777643507741.872049847804311.597830464
507765.093801112804494.499658468507781.822069432804588.501690309
 507797.55087196804644.673412022507907.788054275804972.599372506
#Sta/Elev= 30
9687.466926.66349709.509911.06689739.656 909.9219759.754898.84649779.852884.6526
 9799.95876.10779850.301866.07469880.542862.09199890.623859.19899900.703  860.83
9910.784856.75789920.864850.50049951.106 841.7959971.267833.51369991.428831.7967
10021.69832.006410052.09 836.67410062.31839.596610082.74839.204710124.06845.4283
10134.44848.960710165.81 853.05110176.39855.685610208.16853.916710282.27861.2937
10324.62866.969210377.56878.704510409.13887.8538 10451.1892.175810500.88 902.801
#Mann= 3 , 0 , 0
9687.466  0.0811       09687.466  0.0811       010500.88  0.0811       0
#XS Ineff= 2 , 0
       0                               0
Bank Sta=9687.466,10500.88
Exp/Cntr=0.3,0.1

Type RM Length L Ch R = 1 ,34180.55,247.787900,247.787900,247.787900
XS GIS Cut Line= 6
 507482.82582328804570.969388576507526.689248549804605.892173552
507669.981654012804699.833989928507721.664781853804747.851214398
 507805.06811817804859.142553385 507876.15203756805008.814286397
#Sta/Elev= 30
9888.986880.47359895.028880.44419905.212878.20849910.666 872.9599927.141854.3488
9943.616839.9123 9978.41 831.2839990.181831.554910001.89830.150410013.54830.0939
10025.19831.168210039.38833.870310048.49835.847110060.79839.5662 10073.2 841.354
 10085.6845.1033 10110.4 846.43210149.85851.881110196.55854.879910249.05 860.621
10261.28 864.11410285.76867.794510297.99871.7267 10321.6881.124910344.57886.3451
10367.38889.375510412.07891.220310423.08892.859110456.03899.845710492.38911.0003
#Mann= 3 , 0 , 0
9888.986  0.0688       09888.986  0.0688       010492.38  0.0688       0
#XS Ineff= 2 , 0
       0                               0
Bank Sta=9888.986,10492.38
Exp/Cntr=0.3,0.1

Type RM Length L Ch R = 1 ,33932.76,470.641600,470.641600,470.641600
XS GIS Cut Line= 6
507369.432741702804818.111861065507550.458232641804896.342429414
507606.420107335804930.674618647507658.366649419804972.051153883
507736.710629493805060.982212603 507861.13097626805263.636823773
#Sta/Elev= 30
9896.527877.36149902.541877.78159913.343874.03079934.947855.34279945.749842.1522
9956.551834.15679967.353827.96439978.155827.897310021.42829.226910043.37834.9475
10065.56 837.56210087.75842.039510110.87842.1638 10208.4852.947110235.43858.4445
10264.12862.485410311.68873.313110341.82881.479310361.48887.975910396.92910.4186
10408.61919.5826   10432940.974710443.69 945.28910455.39945.789210478.78968.6878
10490.47978.440210532.021004.71310551.311013.58110572.331017.48810582.431017.381
#Mann= 3 , 0 , 0
9896.527    0.12       09896.527    0.12       010582.43    0.12       0
#XS Ineff= 2 , 0
       0                               0
Bank Sta=9896.527,10582.43
Exp/Cntr=0.3,0.1

Type RM Length L Ch R = 1 ,33462.12,382.235400,382.235400,382.235400
XS GIS Cut Line= 6
507343.757533431804868.376032665507281.053013086804924.113384068
 507236.75402936804978.104381456507154.063573798805103.348316215
507044.234398654805308.295968112506984.020509619805462.994935174
#Sta/Elev= 30
9690.746877.18979702.464875.78269742.602862.32489784.185861.7199 9801.66858.3212
9840.465840.3521 9864.41839.34469912.597832.61559955.048832.38979992.835825.7739
10019.55826.627710031.05829.706810042.55 835.33610065.55850.668310077.06860.1281
10088.56  872.4110100.06887.266810123.06910.852810135.16913.617610145.49922.1742
 10167.8945.791610180.33956.979610201.25980.618610212.41989.840210234.531004.273
10267.171020.62810293.761029.40510331.681033.04910363.671042.70910393.311044.144
#Mann= 3 , 0 , 0
9690.746    0.12       09690.746    0.12       010393.31    0.12       0
#XS Ineff= 2 , 0
       0                               0
Bank Sta=9690.746,10393.31
Exp/Cntr=0.3,0.1

Type RM Length L Ch R = 1 ,33079.89,386.062200,386.062200,386.062200
XS GIS Cut Line= 3
507258.160886616804767.849738151506959.567932665804768.845047981
506750.401638279804774.313785736
#Sta/Elev= 30
 9785.85861.82139809.011861.03989819.011 858.8619859.011841.69569879.011835.6242
9889.011833.51499909.011831.54619919.011828.77949939.011829.11459979.012 824.712
10029.01822.678610039.01825.503810049.01832.577910059.01 843.42710079.01870.1225
10089.01880.599710109.02895.346310119.02899.900410129.03902.393210139.03913.6662
10149.03922.537110169.04935.864110179.04947.881710209.05964.430610219.06971.7356
10229.06977.226810239.07981.497210249.07987.925310259.07992.145910293.681000.551
#Mann= 3 , 0 , 0
 9785.85  0.0855       0 9785.85  0.0855       010293.68  0.0855       0
#XS Ineff= 2 , 0
       0                               0
Bank Sta=9785.85,10293.68
Exp/Cntr=0.3,0.1

Type RM Length L Ch R = 1 ,32693.82,66.629500,66.629500,66.629500
XS GIS Cut Line= 2
507217.238658965804202.670903146506705.085881144804610.657014236
#Sta/Elev= 30
 9700.41875.88989741.627872.55949792.768 851.5669805.553849.94659818.338 851.179
9832.543848.24959848.592849.42739880.691847.92279928.839 823.1519944.889818.9141
9993.037817.479810010.11818.6381 10022.9829.550910041.18833.554710048.47833.6462
10074.04825.203310086.82819.295210099.61822.1314 10112.4832.988710137.48849.7856
10153.53852.845510163.54859.466410176.32873.730210189.11882.500810214.68893.8389
10240.25900.300510253.03901.731610265.88906.073910314.02933.1113 10355.2959.4371
#Mann= 3 , 0 , 0
 9700.41  0.0644       0 9700.41  0.0644       0 10355.2  0.0644       0
#XS Ineff= 2 , 0
       0                               0
Bank Sta=9700.41,10355.2
Exp/Cntr=0.3,0.1

Type RM Length L Ch R = 3 ,32659.37,,,
BEGIN DESCRIPTION:
END DESCRIPTION:
Bridge Culvert--1,0,-1,-1, 0
Deck Dist Width WeirC Skew NumUp NumDn MinLoCord MaxHiCord MaxSubmerge Is_Ogee
22.980150,20.669200,2.6,0, 60, 60, , , 0.95, 0, 0,0,,
 9721.65 9722.04 9731.22 9738.57 9743.77 9755.11 9756.33 9768.88 9771.64 9781.44
 9788.18 9794.00 9804.71 9806.55 9819.11 9821.25 9831.67 9837.79 9844.22 9854.32
 9856.78 9869.33 9870.86 9881.89 9887.39 9889.28 9929.99 9929.9910092.3910092.39
10165.2310167.2810169.0910182.2610182.6510195.4210198.0310198.7410208.3210213.99
10221.1410229.9910233.9510245.9810246.7610259.5810261.9810272.3910277.9710285.20
10293.9610298.0210309.9610310.8310323.6410325.9510336.4610341.9510349.2710355.34
  870.17  869.86  864.90  864.88  863.96  861.28  860.96  860.80  860.06  860.13
  860.50  860.80  858.42  858.04  854.73  854.25  853.13  852.27  852.07  851.95
  851.85  850.33  850.17  849.12  848.42  848.39  848.45  848.45  848.68  848.68
  848.78  848.79  848.75  848.86  848.86  857.85  859.09  859.64  866.98  869.77
  870.66  875.12  876.56  886.37  886.96  893.17  894.65  900.62  904.09  907.42
  911.27  913.17  921.48  922.07  931.24  933.05  942.18  947.09  952.96  955.79
 -129.83 -130.14 -135.10 -135.12 -136.04 -138.72 -139.04 -139.20 -139.94 -139.87
 -139.50 -139.20 -141.58 -141.96 -145.27 -145.75 -146.87 -147.73 -147.93 -148.05
 -148.15 -149.67 -149.83 -150.88 -151.58 -151.61 -151.55  843.45  843.68 -151.32
 -151.22 -151.21 -151.25 -151.14 -151.14 -142.15 -140.91 -140.36 -133.02 -130.23
 -129.34 -124.88 -123.44 -113.63 -113.04 -106.83 -105.35  -99.38  -95.91  -92.58
  -88.73  -86.83  -78.52  -77.93  -68.76  -66.95  -57.82  -52.91  -47.04  -44.21
 9721.65 9722.04 9731.22 9738.57 9743.77 9755.11 9756.33 9768.88 9771.64 9781.44
 9788.18 9794.00 9804.71 9806.55 9819.11 9821.25 9831.67 9837.79 9844.22 9854.32
 9856.78 9869.33 9870.86 9881.89 9887.39 9889.28 9945.84 9945.8410108.2410108.24
10165.2310167.2810169.0910182.2610182.6510195.4210198.0310198.7410208.3210213.99
10221.1410229.9910233.9510245.9810246.7610259.5810261.9810272.3910277.9710285.20
10293.9610298.0210309.9610310.8310323.6410325.9510336.4610341.9510349.2710355.34
  870.17  869.86  864.90  864.88  863.96  861.28  860.96  860.80  860.06  860.13
  860.50  860.80  858.42  858.04  854.73  854.25  853.13  852.27  852.07  851.95
  851.85  850.33  850.17  849.12  848.42  848.39  848.47  848.47  848.70  848.70
  848.78  848.79  848.75  848.86  848.86  857.85  859.09  859.64  866.98  869.77
  870.66  875.12  876.56  886.37  886.96  893.17  894.65  900.62  904.09  907.42
  911.27  913.17  921.48  922.07  931.24  933.05  942.18  947.09  952.96  955.79
 -129.83 -130.14 -135.10 -135.12 -136.04 -138.72 -139.04 -139.20 -139.94 -139.87
 -139.50 -139.20 -141.58 -141.96 -145.27 -145.75 -146.87 -147.73 -147.93 -148.05
 -148.15 -149.67 -149.83 -150.88 -151.58 -151.61 -151.53  843.47  843.70 -151.30
 -151.22 -151.21 -151.25 -151.14 -151.14 -142.15 -140.91 -140.36 -133.02 -130.23
 -129.34 -124.88 -123.44 -113.63 -113.04 -106.83 -105.35  -99.38  -95.91  -92.58
  -88.73  -86.83  -78.52  -77.93  -68.76  -66.95  -57.82  -52.91  -47.04  -44.21
Pier Skew, UpSta & Num, DnSta & Num=  ,10011.19, 2 ,10027.04, 2 , 0 , 0 , 0 ,,
    4.00    4.00
 -151.44  848.56
    4.00    4.00
 -151.41  848.59
BR Coef=-1 , 0 , 0 ,, 0 ,,,0.8,0,1,0,
WSPro=,,,, 1 ,,,, 0 ,,,, 0 ,,,,-1 ,-1 ,-1 , 0 , 0 , 0 , 0 , 0
BC Design=,, 0 ,, 0 ,,,,,,

Type RM Length L Ch R = 1 , 32627.2,245.785500,245.785500,245.785500
XS GIS Cut Line= 2
507173.070552695804147.760838146506686.264699669804558.340863649
#Sta/Elev= 30
9711.321882.45719722.549873.8329 9734.96871.14899748.042876.7461 9753.57877.7686
9761.124876.86419774.206874.17769813.452860.13579831.123857.62779846.634853.3132
9905.025848.60629918.106844.0715 9944.27827.38669970.718817.378910032.76818.7783
10048.27824.690410062.01827.4204 10094.8820.514810110.31 820.67710127.42826.7481
10141.33839.693110153.58 848.01610156.84849.255410205.91850.083610218.89860.9298
 10234.4879.023210271.32902.266210311.95925.506510336.73941.236710348.15 946.176
#Mann= 3 , 0 , 0
9711.321  0.0802       09711.321  0.0802       010348.15  0.0802       0
#XS Ineff= 2 , 0
       0                               0
Bank Sta=9711.321,10348.15
Exp/Cntr=0.3,0.1

Type RM Length L Ch R = 1 ,32381.41,245.785600,245.785600,245.785600
XS GIS Cut Line= 6
506855.199941746803904.970272742506798.379228848804075.632081054
506757.724878302804176.055141829506664.888979703804358.333437758
506623.714546911804425.234466322506557.738017135804520.347970523
#Sta/Elev= 30
9677.4491045.3559729.8211009.5289761.537994.37649775.297981.76859803.824966.5116
9824.968951.8826 9835.54939.23749846.112920.24119856.683905.01789878.246884.3016
9899.823860.75879932.188835.96729942.977829.60659953.765817.26079964.553813.2148
9986.825815.85719997.981819.527310042.66813.720610053.82814.702510064.99818.7375
 10109.7827.105610143.77847.037810155.13 852.293 10178.1853.605210189.84861.0621
10213.33867.835910248.56882.106510299.66907.639110321.26924.569910364.59951.1427
#Mann= 3 , 0 , 0
9677.449    0.04       09677.449    0.04       010364.59    0.04       0
#XS Ineff= 2 , 0
       0                               0
Bank Sta=9677.449,10364.59
Exp/Cntr=0.3,0.1

Type RM Length L Ch R = 1 ,32135.62,245.785500,245.785500,245.785500
XS GIS Cut Line= 6
506526.976778048803879.722337091506506.658193693804095.281097371
506502.731546301804210.992054595506493.240303654 804285.01499989
 506463.82538203804414.349836549506430.576938671 804506.60082692
#Sta/Elev= 30
9733.8731022.1969759.3031004.5869779.423 985.8869799.544973.41429839.781941.9479
9869.876 912.7249879.908902.10589889.939882.14869910.003849.39359940.098 820.468
9950.129813.80939960.132811.27189970.133809.824110010.14809.516910040.19 811.732
10080.38824.556610090.46829.706110100.54830.4405 10120.7836.433910130.79842.9585
10151.05860.2432 10181.6862.087910232.92888.130310253.59897.304710295.34 909.658
10316.39913.810710326.92920.554110330.84 921.733 10348.4924.845410371.71931.4066
#Mann= 3 , 0 , 0
9733.873  0.0473       09733.873  0.0473       010371.71  0.0473       0
#XS Ineff= 2 , 0
       0                               0
Bank Sta=9733.873,10371.71
Exp/Cntr=0.3,0.1

Type RM Length L Ch R = 1 ,31889.84,245.785500,245.785500,245.785500
XS GIS Cut Line= 6
506272.876893171803839.204787189506257.638940646804017.096312502
506262.969933346804217.366062325506261.896226984804327.281550139
506257.490195935804383.138047633 506242.34679897804486.251622612
#Sta/Elev= 30
9681.345988.69949727.412984.69379757.565972.81599767.616966.3215 9797.77941.3742
9847.838  894.999857.851873.68499897.855 824.1069907.855819.17489927.865821.9429
9947.878 815.1619957.884 807.593 9997.91 799.64110017.93802.525710037.95808.1865
10057.97809.456410097.97823.520510117.97837.085210137.98855.646610157.99870.8248
10178.02878.227210188.05 877.77210198.08 879.89410208.12891.360410218.15906.2263
10228.19916.080610268.54941.010510288.72955.288310319.12972.936110330.55977.3472
#Mann= 3 , 0 , 0
9681.345   0.062       09681.345   0.062       010330.55   0.062       0
#XS Ineff= 2 , 0
       0                               0
Bank Sta=9681.345,10330.55
Exp/Cntr=0.3,0.1

Type RM Length L Ch R = 1 ,31644.05,572.000400,572.000400,572.000400
XS GIS Cut Line= 6
506129.214673719 803780.18077454 506085.08737907803935.564789988
506025.603955749804118.681301413506003.960301872804178.854451658
505963.864157205804304.630860379505941.499314459 804382.98983661
#Sta/Elev= 30
9619.755947.51659635.091934.4934 9645.44931.24099666.137914.38819676.486908.1335
9697.184898.21339718.066894.91329728.508 891.6799746.841881.79649822.767846.1287
9843.796831.8323 9854.31822.97269864.825816.69179896.368810.3066 9948.94 807.347
9980.561798.746210012.47797.770110023.08798.1641 10033.7  801.8210075.73823.4349
10096.72836.4901 10128.2860.0374 10138.7866.210110159.69881.473810170.18890.7478
10180.59896.132910211.81897.858810232.62926.160910243.02929.997710251.29935.9192
#Mann= 3 , 0 , 0
9619.755  0.0524       09619.755  0.0524       010251.29  0.0524       0
#XS Ineff= 2 , 0
       0                               0
Bank Sta=9619.755,10251.29
Exp/Cntr=0.3,0.1

Type RM Length L Ch R = 1 ,31072.05,408.312800,408.312800,408.312800
XS GIS Cut Line= 5
505597.228349209803557.581384704 505582.98595041803650.156976849
505519.519594193803965.708543763505520.829051882804111.250474781
505524.456088126804124.325662747
#Sta/Elev= 30
9705.824 904.4019723.448 895.2939743.683889.10419784.154 885.2079794.271 885.918
9804.429890.28269814.629890.0247 9835.03 884.888 9845.23879.8851 9855.43871.2632
9875.831858.39979916.632822.73469926.832807.45219937.032802.42699947.232 795.836
9957.433791.48249977.833791.396310039.03793.654310059.44798.757910090.04 797.203
10120.64804.194210130.65803.354110140.65804.069710150.65806.979810160.65811.3393
10200.65834.693110220.66843.522510250.66854.937910266.91863.553710280.48868.4227
#Mann= 3 , 0 , 0
9705.824    0.12       09705.824    0.12       010280.48    0.12       0
#XS Ineff= 2 , 0
       0                               0
Bank Sta=9705.824,10280.48
Exp/Cntr=0.3,0.1

Type RM Length L Ch R = 1 ,30663.74,245.785500,245.785500,245.785500
XS GIS Cut Line= 6
505001.825097734803532.263730773505077.313676356803677.419220078
505220.490384505803996.040599126505238.388707064804026.749952585
505263.469649548804061.676068627505314.163362981804112.609858179
#Sta/Elev= 30
9657.259885.1178 9663.93885.36239671.741883.30429683.111877.88389717.221872.4827
9728.591865.9431 9735.03865.02349748.783859.61189784.626838.89369795.812833.7308
9829.269825.00859840.322824.74869862.427818.86489884.533 814.8769895.585810.9651
9909.372803.79219928.543798.16659961.282794.33979972.195790.93629983.108789.8892
10026.64790.8042 10048.4796.757710070.16798.367810091.92 798.028 10102.8800.2205
10146.79804.808310265.65810.782510294.86814.782910309.12820.517510320.76826.7915
#Mann= 3 , 0 , 0
9657.259   0.013       09657.259   0.013       010320.76   0.013       0
#XS Ineff= 2 , 0
       0                               0
Bank Sta=9657.259,10320.76
Exp/Cntr=0.3,0.1

Type RM Length L Ch R = 1 ,30417.95,245.785500,245.785500,245.785500
XS GIS Cut Line= 6
504675.900668453803845.179440524504787.810272162803906.802731152
504905.416740821803961.838888839505042.021275988804013.714879934
 505239.19879114 804094.36370351505312.802167069804128.036745302
#Sta/Elev= 30
9684.098888.20219694.663890.57929717.762890.81869729.126888.2004 9740.49883.4545
9744.918880.18359763.218870.38949774.582862.39569787.021849.95929819.879821.3223
9842.163806.69749853.305802.14099886.552798.3767 9919.39792.34129941.282790.4631
9978.159790.33219994.915788.967910005.61789.597710016.29 793.10410048.33789.1278
10069.69788.757110087.86790.222710101.89793.559410155.91801.115710199.12804.9724
10220.73806.444710329.07809.899110339.99811.590310361.83 821.94510381.87833.8705
#Mann= 3 , 0 , 0
9684.098  0.0332       09684.098  0.0332       010381.87  0.0332       0
#XS Ineff= 2 , 0
       0                               0
Bank Sta=9684.098,10381.87
Exp/Cntr=0.3,0.1

Type RM Length L Ch R = 1 ,30172.17,245.785600,245.785600,245.785600
XS GIS Cut Line= 6
 504699.81511596804271.591072537504810.478205479804262.459119538
504906.632542959804243.346816301505213.681625424804145.049552997
 505265.41397371804139.795469468505311.356344359804144.422735983
#Sta/Elev= 30
9716.817882.70929732.006876.17599742.017 878.0989752.042886.99269762.066890.1672
9782.131889.20499802.272885.55559842.667858.51599862.965849.09919873.114841.5221
9883.325838.78719893.574833.73769914.072813.23449924.321801.30899934.643792.9459
9955.315785.58149998.549782.045810017.53784.276310049.04784.842710070.33787.6045
10091.74787.351310123.86792.702110147.72801.772910177.38  803.2810188.05805.0862
10260.23806.9282 10290.4809.753910300.42813.551510340.63 835.146 10347.1840.3269
#Mann= 3 , 0 , 0
9716.817  0.0426       09716.817  0.0426       0 10347.1  0.0426       0
#XS Ineff= 2 , 0
       0                               0
Bank Sta=9716.817,10347.1
Exp/Cntr=0.3,0.1

Type RM Length L Ch R = 1 ,29926.38,245.785500,245.785500,245.785500
XS GIS Cut Line= 6
504894.478158649804573.831059917504979.966380191804536.278223585
505045.251608064804491.681765444505177.093921597804351.673887571
505224.053469525804307.950981328 505305.12355025804248.001528711
#Sta/Elev= 30
9740.917959.04399752.014947.30779762.625939.42649795.253907.90549806.322898.3871
9817.585883.73319840.371 862.1289852.149860.10969855.788857.92029874.715843.6352
9900.764825.33259926.888810.2994 9940.54799.90779952.774793.31929968.101785.8874
9983.272776.95189993.875772.774610007.04 772.63710020.15 773.36410029.39774.7203
   10060782.6014 10101.5788.0322 10115.9 792.52910130.57799.903610184.31802.4693
10222.81806.852310235.04809.823410247.04814.806610259.05821.2167 10271.2826.5413
#Mann= 3 , 0 , 0
9740.917  0.0531       09740.917  0.0531       0 10271.2  0.0531       0
#XS Ineff= 2 , 0
       0                               0
Bank Sta=9740.917,10271.2
Exp/Cntr=0.3,0.1

Type RM Length L Ch R = 1 , 29680.6,221.867300,221.867300,221.867300
XS GIS Cut Line= 6
504982.338481584804710.245771821505078.392628582804690.884549987
505158.775273199804664.867549992505254.463752717804618.598022152
505337.451827503804563.595415788505428.113558771804520.718504173
#Sta/Elev= 30
9676.592931.50399689.442924.51729709.739914.76789719.887908.91589730.036907.1854
9760.859 891.6029781.505882.1817 9802.33871.92729823.341864.21089855.144 854.198
9858.747852.28899876.777835.51959887.643826.3942 9898.51817.55069909.613809.6852
9932.219795.66899943.522792.54269954.826790.51879966.174786.40479978.323773.4685
 10002.7769.946510014.98769.6478 10038.9770.212510062.27774.8875 10083.6787.2807
10096.27794.045510118.46803.182210129.45 811.26210153.62 826.87810165.51835.3473
#Mann= 3 , 0 , 0
9676.592    0.12       09676.592    0.12       010165.51    0.12       0
#XS Ineff= 2 , 0
       0                               0
Bank Sta=9676.592,10165.51
Exp/Cntr=0.3,0.1

Type RM Length L Ch R = 1 ,29458.73,269.703800,269.703800,269.703800
XS GIS Cut Line= 5
504962.537304043804765.620330352505164.520489812804755.113360852
 505215.77866137804765.000000015505431.323617578  804890.6324099
 505579.59259023 804961.47611856
#Sta/Elev= 30
9652.021926.63019674.514917.78559684.528909.63249704.555 897.1069724.582887.3489
9764.636872.30759784.663867.49249794.677863.07199814.704846.09419834.731832.4159
9854.766815.46429875.135801.20339917.154777.91289928.729772.95679940.303770.2967
9951.878 764.7479963.453763.0754 10032.9763.839410056.05767.928110067.62 773.365
10105.06800.079910155.97829.518610182.21850.507610226.54879.819910237.62 885.728
10259.79 906.06910270.87 913.23610281.95915.905510304.12928.761610320.29944.5148
#Mann= 3 , 0 , 0
9652.021    0.12       09652.021    0.12       010320.29    0.12       0
#XS Ineff= 2 , 0
       0                               0
Bank Sta=9652.021,10320.29
Exp/Cntr=0.3,0.1

Type RM Length L Ch R = 1 ,29189.03,245.785500,245.785500,245.785500
XS GIS Cut Line= 6
504891.870774056804912.475520652504981.901137527804944.062617056
505079.828614478804992.400117363505151.708866407805037.515505064
505363.634355759805188.298617102505452.901204674805254.971866375
#Sta/Elev= 30
9698.751 914.4499722.912902.07419733.505895.23729744.171 891.1449776.171872.3708
9786.838868.43119819.545848.6312 9866.38815.25149897.995784.45299908.353777.8164
9933.182 767.6899964.786759.769410001.21758.1559 10029.2762.291910041.47762.6896
10053.74762.838310066.01759.673810087.47760.413910139.22776.164910151.92783.4768
10164.19786.924710173.73791.697310188.74802.298510250.13837.870410262.61844.6558
10275.09849.101310293.04859.659810300.05862.796410325.01867.867810359.84 881.389
#Mann= 3 , 0 , 0
9698.751  0.0538       09698.751  0.0538       010359.84  0.0538       0
#XS Ineff= 2 , 0
       0                               0
Bank Sta=9698.751,10359.84
Exp/Cntr=0.3,0.1

Type RM Length L Ch R = 1 ,28943.24,245.785500,245.785500,245.785500
XS GIS Cut Line= 6
504789.698209764 805126.39932715504908.359326602805184.019365784
505036.614768891805254.559214597505103.470290907805295.436526152
505210.627152731805368.064091834505357.623199782805477.287211097
#Sta/Elev= 30
9739.871938.88479756.678939.45659767.662934.39329778.646924.8015 9789.63912.3951
 9800.75894.02879823.181 873.7259868.044828.35699879.385808.23429890.789793.2206
9902.193781.18989915.458771.76469947.809755.12739977.866751.950110039.74754.2444
10051.46758.1291 10098.4766.987710110.48775.056710146.72804.754610182.96826.0437
10195.04835.7922 10219.2848.833210231.41852.2771 10288.7848.243610305.66850.1623
10318.03856.591910367.68889.184410380.39 893.121 10393.1894.335610409.15899.7418
#Mann= 3 , 0 , 0
9739.871  0.0502       09739.871  0.0502       010409.15  0.0502       0
#XS Ineff= 2 , 0
       0                               0
Bank Sta=9739.871,10409.15
Exp/Cntr=0.3,0.1

Type RM Length L Ch R = 1 ,28697.46,245.785600,245.785600,245.785600
XS GIS Cut Line= 6
504688.090375706805344.320462907 504753.87431241805376.999340681
504838.621679744 805423.53607414504936.821615348805481.971828089
505112.123432885805592.238507133505264.482220098805694.616163697
#Sta/Elev= 30
9757.068906.12159787.115897.73819809.447 894.2849820.613888.07529866.032845.9286
 9877.44831.70869888.849820.90379900.257803.60839923.074776.60579934.609760.8122
9946.217747.94619981.038747.395510015.95750.563910051.14751.536110074.77756.0282
 10098.4769.361310122.02780.248910145.65794.150410169.28801.882210181.09803.7551
10192.91809.703210216.54817.994210240.16821.794110300.03845.397110325.95859.3565
10348.02863.977810360.02868.925910372.02 877.076 10420.5901.899810432.15 909.437
#Mann= 3 , 0 , 0
9757.068  0.0555       09757.068  0.0555       010432.15  0.0555       0
#XS Ineff= 2 , 0
       0                               0
Bank Sta=9757.068,10432.15
Exp/Cntr=0.3,0.1

Type RM Length L Ch R = 1 ,28451.67,245.785500,245.785500,245.785500
XS GIS Cut Line= 6
504578.988835261805601.029969827504713.959884699805650.323393169
504839.417788801805692.010639032504967.470158431805746.300219306
505100.614854184805812.839613189505190.835085871805866.459476888
#Sta/Elev= 30
9790.348869.98139807.495 851.4689818.176842.5097 9828.81830.30689850.078817.5741
9859.582810.22769892.613780.48479903.247768.69979913.881759.69859924.515754.1883
9935.136750.86089966.667742.98769977.178741.960310051.01742.717710126.62761.7676
10137.48766.641210170.07773.815110191.79782.047410224.73 796.817   10249803.9167
10272.22 806.75410293.89814.292110325.33836.516910347.88 847.98610358.54855.8403
10378.62865.631210398.69866.748810428.61861.733310437.75861.675710459.18 865.414
#Mann= 3 , 0 , 0
9790.348  0.0641       09790.348  0.0641       010459.18  0.0641       0
#XS Ineff= 2 , 0
       0                               0
Bank Sta=9790.348,10459.18
Exp/Cntr=0.3,0.1

Type RM Length L Ch R = 1 ,28205.88,179.343900,179.343900,179.343900
XS GIS Cut Line= 6
504459.201626956805847.069400751 504535.93039497805874.725874236
504598.426220729805892.298362136504658.148705075805904.303197799
504824.362259766805920.329657667504923.005970329805948.672872134
#Sta/Elev= 30
9712.626864.30999734.465854.2101 9764.75838.55599795.218821.11719803.627815.4536
9814.014806.76789845.178779.2501 9865.83773.63819872.834770.6944 9876.03768.8829
 9886.23760.3782 9896.43753.4293 9906.63750.0871 9916.83747.8559 9926.94747.5076
9937.008748.12919947.077747.39529967.203744.58929977.213741.154610017.26740.4659
10027.27740.480910037.29741.3897 10057.5745.698310087.84749.764510098.13752.4152
   10129765.236710139.37771.372310149.84778.716310170.92785.042610189.91788.7712
#Mann= 3 , 0 , 0
9712.626  0.0618       09712.626  0.0618       010189.91  0.0618       0
#XS Ineff= 2 , 0
       0                               0
Bank Sta=9712.626,10189.91
Exp/Cntr=0.3,0.1

Type RM Length L Ch R = 1 ,28026.54,312.227200,312.227200,312.227200
XS GIS Cut Line= 6
504397.921817863 805888.50259038504504.440909572805954.087238845
504558.591672318805989.913323557504608.305261944806025.143670556
504716.011149672806105.192669032504900.110118099806247.982040592
#Sta/Elev= 30
9661.566876.65069693.365 856.2819728.596835.32279752.083819.34479763.826813.2138
 9775.57803.98229799.318 792.0819835.289765.17159847.279755.32999877.679743.3815
9894.974742.05689908.466736.27669912.269733.73129929.106729.67829983.002728.9515
10013.07729.530110032.95732.483110045.45733.083310058.09731.235610070.74731.7666
10079.03734.860210108.71749.536110121.37762.7787 10144.3784.019610171.99807.8017
10225.88848.3359 10242.2862.856410260.57 873.82110273.23875.7291 10279.7880.0791
#Mann= 3 , 0 , 0
9661.566    0.12       09661.566    0.12       0 10279.7    0.12       0
#XS Ineff= 2 , 0
       0                               0
Bank Sta=9661.566,10279.7
Exp/Cntr=0.3,0.1

Type RM Length L Ch R = 1 ,27714.31,245.785500,245.785500,245.785500
XS GIS Cut Line= 6
504245.275122567806072.023044562504344.510854463806159.822524132
504385.715492283806202.079651775504486.788352102806333.553702998
504531.024412952806385.161183316504674.045038231806526.940233159
#Sta/Elev= 30
9680.288856.21129719.435839.70039732.867836.84179759.733828.7201 9775.63822.3911
9786.598816.43099842.155781.0893 9861.94  771.129901.202748.44829915.471736.4177
9928.343734.87649948.757734.27989966.351729.69419982.392728.072510034.74729.1539
10065.81736.005210079.25735.621810092.42737.151610119.56744.0879 10125.8746.7821
10140.11755.272810168.69 775.74410182.67787.411410189.98793.734810218.59822.6716
 10247.2848.038210266.58866.473910280.56874.302210294.55876.6011 10307.2886.5217
#Mann= 3 , 0 , 0
9680.288  0.0668       09680.288  0.0668       0 10307.2  0.0668       0
#XS Ineff= 2 , 0
       0                               0
Bank Sta=9680.288,10307.2
Exp/Cntr=0.3,0.1

Type RM Length L Ch R = 1 ,27468.53,245.785500,245.785500,245.785500
XS GIS Cut Line= 6
504053.654640524806275.622245706504119.026353495806336.992843664
504179.508575436806387.118919584 504404.34950402 806542.00117742
504499.722280926806623.587206273504547.132660522806669.808292658
#Sta/Elev= 30
9661.495850.16879691.031830.3154 9732.01811.98939758.928798.38859771.916789.9144
9810.731759.8066  9836.5733.7683 9848.84725.01419885.861724.47569921.895727.4411
9933.816731.12219949.527 733.048  9967.9733.21269981.497731.46469993.418722.7625
10005.41722.1208 10029.6722.642110040.05728.4474 10041.7730.109610053.91756.3166
10057.39759.4406 10139.3817.402410155.15 831.90110185.47 849.92710215.49876.6191
10228.38880.280810235.75884.114310263.68910.434110277.64919.138210294.59  922.04
#Mann= 3 , 0 , 0
9661.495  0.0992       09661.495  0.0992       010294.59  0.0992       0
#XS Ineff= 2 , 0
       0                               0
Bank Sta=9661.495,10294.59
Exp/Cntr=0.3,0.1

Type RM Length L Ch R = 1 ,27222.74,293.469700,293.469700,293.469700
XS GIS Cut Line= 6
503969.056945061806379.322646579504115.775789438806566.490123091
 504143.43834052806618.178490669504159.884143442806685.296651235
504183.718023563806733.645333665504309.246792303806914.490899935
#Sta/Elev= 30
  9665.6848.63539672.906847.07939698.643832.80789706.818831.5651 9737.25821.6226
9775.856 800.0599788.725791.61629802.146 778.5669818.034 769.0779851.199734.3064
9864.535727.88269868.189724.43149885.179719.16799936.544 720.417 9962.18723.6782
9981.821719.476310000.27718.481310041.96720.327210052.81  724.2210087.71730.7118
10111.02740.426210141.97765.322610159.02770.156510220.17780.181110244.75785.9583
10257.04797.826510263.84798.986210281.61807.871410298.25812.813910305.56819.0919
#Mann= 3 , 0 , 0
  9665.6  0.0678       0  9665.6  0.0678       010305.56  0.0678       0
#XS Ineff= 2 , 0
       0                               0
Bank Sta=9665.6,10305.56
Exp/Cntr=0.3,0.1

Type RM Length L Ch R = 1 ,26929.27,365.250400,365.250400,365.250400
XS GIS Cut Line= 6
503769.211488273806585.792032701503773.051412361806593.149225047
503804.337385004806646.253190492503905.616379845806802.513757702
504026.983184217806989.758762874504028.775216179806992.640879301
#Sta/Elev= 30
9732.581 848.3619743.028843.65949766.241827.6232 9801.06801.49449824.855791.0368
9848.689776.96499872.522765.90439908.272740.43659920.189732.87269932.435726.8279
9955.939720.42059967.856716.45899979.773714.66659987.593  714.5210027.44715.0865
10039.36719.065410063.19722.858910075.11721.590810087.03721.8946 10097.9727.4656
10098.94728.080510110.86743.168210122.78752.398710146.61778.717110158.53789.6978
10170.44803.138510182.36815.643910194.28824.983910206.19832.737110215.26832.9164
#Mann= 3 , 0 , 0
9732.581  0.0649       09732.581  0.0649       010215.26  0.0649       0
#XS Ineff= 2 , 0
       0                               0
Bank Sta=9732.581,10215.26
Exp/Cntr=0.3,0.1

Type RM Length L Ch R = 1 ,26564.02,296.740400,296.740400,296.740400
XS GIS Cut Line= 6
 503598.20123584 806693.40517075503578.689811547806790.689660177
503575.207216162806841.482342123  503579.9386844806908.288324739
503600.068782397807020.498927834 503656.30245477807274.911009377
#Sta/Elev= 30
9703.234 824.9979745.877813.48819766.306804.96179776.446802.97839806.815 790.193
9836.885756.33249846.909750.21889856.925750.68499866.929748.32669886.968732.0561
9917.116728.31859927.232723.69049947.528721.46649967.823714.84829977.971714.1402
9988.119709.86979998.267709.746310069.78710.297510080.02711.732310090.27716.6978
   10121721.078310141.49726.570910151.74730.000410161.98735.552110182.47749.2025
10213.21 774.00110243.94791.511110254.19795.886610264.43795.531610294.99800.1067
#Mann= 3 , 0 , 0
9703.234  0.0894       09703.234  0.0894       010294.99  0.0894       0
#XS Ineff= 2 , 0
       0                               0
Bank Sta=9703.234,10294.99
Exp/Cntr=0.3,0.1

Type RM Length L Ch R = 1 ,26267.28,273.467200,273.467200,273.467200
XS GIS Cut Line= 6
503426.627910967806839.787801099503343.539672384806946.634730026
 503312.61290297807000.287545261503295.562427968807073.831069781
503261.632413704807184.783451176503232.398172585807298.671850698
#Sta/Elev= 30
9763.794782.15119782.906780.16549808.278757.99839833.649738.3266 9859.02724.2357
9880.525716.27269896.777708.52719909.099706.5244 9935.36706.51239961.183709.7838
 9966.12709.52619976.597706.44979997.033705.479210048.44705.766910058.89709.3593
10069.35710.527710090.27718.091310100.72728.109410111.18746.985310121.64762.4745
10141.27783.682310173.77814.427210184.15827.931510204.92841.7386 10215.3852.9041
10235.86870.183610246.12877.716110256.38  880.9310266.63882.5197 10270.4885.2779
#Mann= 3 , 0 , 0
9763.794  0.0406       09763.794  0.0406       0 10270.4  0.0406       0
#XS Ineff= 2 , 0
       0                               0
Bank Sta=9763.794,10270.4
Exp/Cntr=0.3,0.1

Type RM Length L Ch R = 1 ,25993.81,245.785500,245.785500,245.785500
XS GIS Cut Line= 6
503383.875784641806789.134133328503299.993225742806823.206102318
503143.435725985806821.711455931503065.784310982806841.539595632
502979.437306479806900.397922167502898.510374043806995.778340805
#Sta/Elev= 30
9812.183776.09869845.504758.59859877.807744.20189898.394731.21249938.574713.6019
9948.595707.85179968.632703.3057 9978.65699.98949988.669695.47679998.687693.3644
10008.71693.511710028.75 701.36510048.75703.601410058.75709.319510068.85721.5194
10078.96744.079110089.07 758.11410099.26769.442110109.66779.266410141.72812.8126
   10153 821.08110164.28826.368410175.91833.845410199.95842.297210212.51844.9206
 10225.5849.829310265.74875.541810333.29 913.67710345.95923.277610371.11935.2999
#Mann= 3 , 0 , 0
9812.183  0.0405       09812.183  0.0405       010371.11  0.0405       0
#XS Ineff= 2 , 0
       0                               0
Bank Sta=9812.183,10371.11
Exp/Cntr=0.3,0.1

Type RM Length L Ch R = 1 ,25748.03,245.785600,245.785600,245.785600
XS GIS Cut Line= 6
503221.818747481806282.139348008503194.299657478806378.128663335
503081.445539696806691.949667145503045.407635464806749.273759796
502925.327969205806892.213967204502873.422085482806968.745823919
#Sta/Elev= 30
9626.881903.55489640.116898.95359650.538890.51659660.961885.46679724.272860.5711
 9776.42824.24159787.015810.99639797.638801.06949861.754749.33229883.127736.0854
9917.606 722.699 9925.76718.17579936.302707.64029957.385697.090510010.11693.5015
10031.26698.360510063.81712.103310075.26732.011610086.71744.408110098.28753.0356
10111.67758.388710144.14 781.88910174.88798.877710205.62812.006810227.85826.4736
10267.11848.179410318.27870.230110366.96894.806110391.12 914.35310407.36924.2425
#Mann= 3 , 0 , 0
9626.881    0.12       09626.881    0.12       010407.36    0.12       0
#XS Ineff= 2 , 0
       0                               0
Bank Sta=9626.881,10407.36
Exp/Cntr=0.3,0.1

Type RM Length L Ch R = 1 ,25502.24,245.785500,245.785500,245.785500
XS GIS Cut Line= 6
502904.123201478806261.297228542502882.060688745 806451.20257693
502861.913169007806585.276807611 502830.90835133806738.041830739
502812.022057341806806.915597382502788.309650089806877.037561606
#Sta/Elev= 30
9672.217881.89789696.079871.34569706.147 865.2069716.214861.55439726.281860.9592
9746.416855.5746 9766.55843.33229826.954791.35859867.235762.06929887.432745.7982
9907.629733.30139927.826707.49239948.023 692.9579958.121693.97449998.719692.2079
10019.08692.602710029.27 697.09410039.45698.619810049.63706.227610059.81723.1502
   10070729.571110090.36739.244610131.29777.453110151.78793.190210182.85811.2528
10193.22820.900710234.84838.097510266.51855.188510277.07 856.09210300.33870.0129
#Mann= 3 , 0 , 0
9672.217  0.0957       09672.217  0.0957       010300.33  0.0957       0
#XS Ineff= 2 , 0
       0                               0
Bank Sta=9672.217,10300.33
Exp/Cntr=0.3,0.1

Type RM Length L Ch R = 1 ,25256.46,245.785500,245.785500,245.785500
XS GIS Cut Line= 6
502615.030231459 806265.88600585502614.704708056 806498.66635642
502618.259875936806626.216589921502616.521637626 806726.14982186
502610.459277337806819.903554419502604.981983887 806872.67021181
#Sta/Elev= 30
9694.549870.15579753.666836.51839783.667817.37619793.667808.88199823.669788.3039
 9853.67765.2087 9863.67760.0488 9873.67757.17999893.671745.58449903.671 737.479
9913.671 726.3339923.672717.27419933.675 712.2559953.683695.04919963.687689.4669
10013.71689.597510023.71691.595310043.72699.655710053.72 705.39510073.72725.8714
10103.73748.499810133.73765.628610163.76779.547510203.84804.144210223.88813.4315
10243.92816.092210253.96814.234910264.01810.326710274.07809.773610301.89815.1132
#Mann= 3 , 0 , 0
9694.549   0.108       09694.549   0.108       010301.89   0.108       0
#XS Ineff= 2 , 0
       0                               0
Bank Sta=9694.549,10301.89
Exp/Cntr=0.3,0.1

Type RM Length L Ch R = 1 ,25010.67,245.785600,245.785600,245.785600
XS GIS Cut Line= 6
502359.574461727 806269.94085936502360.596072415806378.762239792
502364.959472271806486.968828449502378.737241381806689.172113963
502383.599718977806788.775512179502385.660731028 806889.54107743
#Sta/Elev= 30
9686.321882.41319701.381873.38389721.382856.76259761.384831.71139791.385807.1591
9811.398788.08939821.407782.19899831.415773.23289841.423760.85449851.431753.8638
9861.439750.12519871.447735.91629881.455716.80139891.463706.36069921.513689.9749
9941.557688.63539961.601690.91399971.623689.90649981.646686.21039991.668686.0069
10041.79689.596210071.86  701.5310111.95727.772610131.97736.722110172.02742.8335
10192.04743.808410232.07754.720210252.07767.392610272.07784.532810306.62798.1541
#Mann= 3 , 0 , 0
9686.321  0.1052       09686.321  0.1052       010306.62  0.1052       0
#XS Ineff= 2 , 0
       0                               0
Bank Sta=9686.321,10306.62
Exp/Cntr=0.3,0.1

Type RM Length L Ch R = 1 ,24764.89,245.785500,245.785500,245.785500
XS GIS Cut Line= 6
502148.025125999806273.298785321502136.375745354 806433.32619727
502126.745225197806601.673938595502124.293663843806640.434643375
502120.968361802806808.389052182502123.263980818 806909.72544285
#Sta/Elev= 30
9669.926840.20089681.658837.48499701.711830.31679721.764827.81789741.817819.7555
9771.896800.92819781.923798.34959791.949793.33219812.002782.2306 9842.07763.0203
9912.184 713.5579922.201702.02279942.233691.47329962.266 685.1619992.315684.0653
10032.39 684.25510042.41686.111310052.41692.508810082.41702.182910102.42712.9123
10122.42728.801310132.42735.328610172.43759.271810192.43768.874510212.44781.5745
10242.45796.745610272.45808.063910282.46809.491710292.46814.004610307.19 824.727
#Mann= 3 , 0 , 0
9669.926    0.12       09669.926    0.12       010307.19    0.12       0
#XS Ineff= 2 , 0
       0                               0
Bank Sta=9669.926,10307.19
Exp/Cntr=0.3,0.1

Type RM Length L Ch R = 1 , 24519.1,245.785500,245.785500,245.785500
XS GIS Cut Line= 6
501975.005716125806223.459663889501931.600085984 806425.68340165
501856.545729066806640.619005443501839.923133662806705.532036505
501831.337663839806755.732738044501827.816601713 806856.48987396
#Sta/Elev= 30
9653.144829.87829664.821831.67659685.059831.64519695.223829.51199705.427825.1417
9736.041805.1763 9756.45793.11229787.138772.68999806.083 758.7529869.866727.1088
9890.828712.06889932.752686.80039943.309683.26969986.136679.001710018.32679.1267
10029.06680.801510039.76687.607710050.31698.892710061.19713.377710071.39729.6228
10081.94743.050410113.03757.465410133.68761.282610154.87761.939610184.77769.0572
10194.91773.361210225.12790.572610245.17798.021910265.22807.758710306.76 817.493
#Mann= 3 , 0 , 0
9653.144  0.0614       09653.144  0.0614       010306.76  0.0614       0
#XS Ineff= 2 , 0
       0                               0
Bank Sta=9653.144,10306.76
Exp/Cntr=0.3,0.1

Type RM Length L Ch R = 1 ,24273.32,245.785600,245.785600,245.785600
XS GIS Cut Line= 6
 501735.64276861806135.772247449501720.657637803806236.781284427
501702.799558221806318.313324031501630.770060866806551.660295561
 501614.73764192806616.711186175501608.507616836806689.555034959
#Sta/Elev= 30
9658.037817.55159667.331814.38499717.903783.10859738.131772.2371 9758.36763.0941
9768.575759.81479799.286745.67029850.576704.99089860.968703.61539871.361 706.168
9892.147716.9032 9902.54712.70699912.933705.36869943.097690.37429954.853688.4418
9965.358682.65099975.863  679.5910017.88678.561310038.88680.091610059.88683.0291
10073.99682.861810101.61684.367710122.21687.410110132.51 689.895 10153.1698.4278
 10173.3710.331310183.38717.176310193.45722.969610203.53730.2508 10228.1749.7896
#Mann= 3 , 0 , 0
9658.037  0.1136       09658.037  0.1136       0 10228.1  0.1136       0
#XS Ineff= 2 , 0
       09910.047                       0
Bank Sta=9658.037,10228.1
Exp/Cntr=0.3,0.1

Type RM Length L Ch R = 1 ,24027.53,245.785500,245.785500,245.785500
XS GIS Cut Line= 6
501371.759422563 806099.36474081501393.695450829806227.100766818
501435.155703107806528.604588398501444.790691238806576.415864627
501453.615694375806607.501058166501462.422199947806630.834426195
#Sta/Elev= 30
9672.163775.11939688.027768.62519708.319762.83099728.612761.53269738.759762.9624
9748.905766.65549759.051766.8133 9789.49756.23579799.637752.53729809.743 746.892
9840.027724.02349870.312710.31269890.502 699.6549900.597692.79329910.692688.6241
9940.977682.81069971.262678.657210011.64677.872810052.01678.5775 10062.1681.7011
10092.38682.632310102.47686.376110112.63692.335810122.83701.699410133.04 707.507
 10174.2724.5179 10184.6730.618510195.21730.4515 10205.9733.231810212.14736.4076
#Mann= 3 , 0 , 0
9672.163   0.077       09672.163   0.077       010212.14   0.077       0
#XS Ineff= 2 , 0
       0                               0
Bank Sta=9672.163,10212.14
Exp/Cntr=0.3,0.1

Type RM Length L Ch R = 1 ,23781.75,245.785500,245.785500,245.785500
XS GIS Cut Line= 6
500973.971350005806320.673753515501026.925848626806378.030857579
501078.024735545806426.162144074501141.026171517806478.104245345
501299.148683939806584.577608821501393.796536982806654.652997667
#Sta/Elev= 30
9685.481787.11949704.497779.12619717.415770.7759 9731.87766.06369745.519758.4151
9760.781754.24479788.394737.34269802.132733.5027 9815.87   726.19842.803698.3604
9847.656695.94339868.724692.98019894.645683.0839 9920.31682.20899932.626678.1439
9961.489677.89749979.637675.918710028.61674.695810045.58675.500810052.41676.9109
10071.72689.375810125.74717.708310140.74723.7084 10157.7728.944510162.88731.3145
10175.27739.472110187.65745.673210200.03749.509910212.63749.552910223.89 758.077
#Mann= 3 , 0 , 0
9685.481  0.0682       09685.481  0.0682       010223.89  0.0682       0
#XS Ineff= 2 , 0
       0                               0
Bank Sta=9685.481,10223.89
Exp/Cntr=0.3,0.1

Type RM Length L Ch R = 1 ,23535.96,245.785600,245.785600,245.785600
XS GIS Cut Line= 6
 500921.43911907 806767.10150543501004.628850666806777.852996996
501085.023152498806775.426612726501255.060652154806740.097583063
501307.853700538806735.262546472501353.224331107806736.289701589
#Sta/Elev= 30
9749.481799.79919753.109796.28049773.488782.06249793.651767.1228 9813.74753.6459
9843.827738.61619853.827733.01729863.827 727.1649883.848714.46549893.871709.1628
9903.893702.20449913.915692.59449924.014675.88899934.112666.75659944.211662.9252
9954.309661.252710016.27660.508410047.13661.510110057.29 662.72410067.46 661.446
10077.62661.737610087.85667.377910097.83674.463610107.87 677.06710127.95676.0862
10137.99680.025810148.01688.490710158.01698.360810168.01710.183410186.24723.1269
#Mann= 3 , 0 , 0
9749.481    0.12       09749.481    0.12       010186.24    0.12       0
#XS Ineff= 2 , 0
       0                               0
Bank Sta=9749.481,10186.24
Exp/Cntr=0.3,0.1

Type RM Length L Ch R = 1 ,23290.17,245.785500,245.785500,245.785500
XS GIS Cut Line= 6
 500927.72838224806994.772833172501037.918505423 807008.69571084
501115.506988813 807006.47698653501365.778144461806986.974615549
501459.326658023 806996.43437027501496.590974968807005.932057268
#Sta/Elev= 30
9682.941 781.4639741.097753.57019751.206745.51669791.278727.80589821.295709.9659
9831.299705.69159841.303699.41059861.311675.29869871.315668.77489881.369 664.941
9901.483660.99839921.597655.16129931.654654.97539941.711 656.7999981.939653.2949
10002.03652.989910022.08 654.25910032.11656.234510042.14660.225710082.22680.8025
10092.22690.854610102.23704.579210112.23716.536610122.23726.572210163.39757.8679
10172.37764.039910202.66776.597210212.76785.923610222.98793.088110255.58804.4005
#Mann= 3 , 0 , 0
9682.941    0.12       09682.941    0.12       010255.58    0.12       0
#XS Ineff= 2 , 0
       0                               0
Bank Sta=9682.941,10255.58
Exp/Cntr=0.3,0.1

Type RM Length L Ch R = 1 ,23044.39,245.785500,245.785500,245.785500
XS GIS Cut Line= 6
500931.364355189807126.395054282501032.047530314807174.017572448
501226.143653344807241.187941105 501318.46520199807278.483758393
501409.131003687807323.977760044501512.429525696807392.845225225
#Sta/Elev= 30
  9701.3779.49729739.466760.09929772.696740.49369805.172725.81869826.497713.7295
9847.654706.11159858.232700.32179889.967680.47069900.545 670.1049911.124662.9541
9942.858657.76749953.437653.89239964.015652.33169974.593653.29649985.171650.6282
 9995.75 650.30410049.31651.024710060.09652.789110103.23666.150910124.98 667.657
10136.04673.831710169.24704.110910200.11723.820210214.55734.605510237.71741.4188
10261.01741.7466   10273744.4672 10297.1752.923810321.48765.6778 10343.5773.3664
#Mann= 3 , 0 , 0
  9701.3  0.1153       0  9701.3  0.1153       0 10343.5  0.1153       0
#XS Ineff= 2 , 0
       0                               0
Bank Sta=9701.3,10343.5
Exp/Cntr=0.3,0.1

Type RM Length L Ch R = 1 , 22798.6,245.785600,245.785600,245.785600
XS GIS Cut Line= 6
500914.945446149807223.219179921501072.110139096 807426.77949219
501092.157588083807458.833778959501167.462775851807566.491922484
501224.738705569807654.807996654501254.430328157807704.443991136
#Sta/Elev= 30
9722.926798.76269725.249797.32179738.582784.26559754.325780.68729776.507 767.972
9801.679756.56739814.265749.00319839.437736.3083 9864.61716.94719886.072695.4295
9914.954671.7432 9927.54665.35029951.946655.17039968.414650.824910037.67649.4753
10062.08650.475210075.24653.003110110.14655.691710127.58663.5326 10135.3668.0857
10159.47685.616710171.39   692.610183.31696.922310207.14711.4617 10242.9741.6029
10254.81749.694110278.12768.013210289.77777.739710301.42790.107210312.43 799.079
#Mann= 3 , 0 , 0
9722.926  0.0643       09722.926  0.0643       010312.43  0.0643       0
#XS Ineff= 2 , 0
       0                               0
Bank Sta=9722.926,10312.43
Exp/Cntr=0.3,0.1

Type RM Length L Ch R = 1 ,22552.82,245.785500,245.785500,245.785500
XS GIS Cut Line= 6
500811.794464993807239.078869535 500827.53155841807299.134359189
500835.406044279807344.761372333500858.576663211807664.642238345
500874.455751454807778.499073244500904.982476001 807938.13724227
#Sta/Elev= 30
9750.722784.73839777.526766.46839787.862750.74529798.198  749.599808.533745.1576
9859.348 705.8099879.443682.62059899.537663.91519919.632648.85969939.682642.5412
9969.717638.03359979.728638.4164 9989.74641.370510009.76642.178410029.79 646.052
10039.81643.912710069.85648.964110109.96651.2916   10120654.404410140.09 663.932
10180.27690.034910301.48748.070210311.65754.536710352.35787.227410362.53791.0255
10382.88 793.682 10413.4792.278110433.75   780.610443.93777.600510457.41770.4659
#Mann= 3 , 0 , 0
9750.722   0.088       09750.722   0.088       010457.41   0.088       0
#XS Ineff= 2 , 0
       0                               0
Bank Sta=9750.722,10457.41
Exp/Cntr=0.3,0.1

Type RM Length L Ch R = 1 ,22307.03,245.785500,245.785500,245.785500
XS GIS Cut Line= 6
500625.642487679 807182.09434406500625.351015455807218.886694331
500619.414511379807305.095600141 500593.01145593807556.097907563
500580.768073826807716.390849432500577.127493305 807861.83666856
#Sta/Elev= 30
9689.586763.41059702.492750.47399712.492735.11889722.493734.97039732.507728.6902
9742.531715.19329752.555 713.0899772.602 700.3699782.626690.86039802.673 666.444
9812.792659.65749883.076639.73529923.293635.15789953.455627.334710003.74623.5483
10033.91625.484410054.02633.216110094.17635.617410124.26640.703910144.32638.2399
10154.34639.763510184.43657.841110224.55673.543110244.56673.581910254.57682.9831
10274.58683.747910284.58686.684610304.59695.847610364.61730.713910371.45736.7368
#Mann= 3 , 0 , 0
9689.586    0.12       09689.586    0.12       010371.45    0.12       0
#XS Ineff= 2 , 0
       0                               0
Bank Sta=9689.586,10371.45
Exp/Cntr=0.3,0.1

Type RM Length L Ch R = 1 ,22061.25,245.785600,245.785600,245.785600
XS GIS Cut Line= 6
500471.978710504807110.384581403500441.360734118807228.139643761
500420.090307242807289.482477649500339.048652939807486.747344643
500303.708790334807587.538054983500273.777894777807700.835587152
#Sta/Elev= 30
9672.458746.80669687.438734.09399707.938722.19939718.188714.1948 9728.47708.1182
9744.944701.74179759.692689.56149790.914669.71939801.442665.0569 9822.61651.0103
9833.194647.07169854.363641.93849908.309635.50229929.928622.47069983.976619.8032
10005.61620.439610016.42622.269710030.42620.187610056.72620.765110059.67621.1391
10070.48626.460110081.12627.774310091.71627.197110102.31630.202310114.83647.8614
 10123.5 658.07310175.27  692.5610228.59 724.91610249.23733.616910296.39762.8871
#Mann= 3 , 0 , 0
9672.458    0.04       09672.458    0.04       010296.39    0.04       0
#XS Ineff= 2 , 0
       0                               0
Bank Sta=9672.458,10296.39
Exp/Cntr=0.3,0.1
